HEC-RAS study Dutchman Creek.prj: Dutchman Creek Limited Detail Study

--- Dutchman Creek.g01 (geometry) --- (continued)

Type RM Length L Ch R =3,124203,,,
BEGIN DESCRIPTION:
Murchison Rd (DC) tor
Structure ID: LDS_DC_10
Approximate Survey Structure
END DESCRIPTION:
Bridge Culvert--1,0,-1,-1,0
Deck Dist Width WeirC Skew NumUp NumDn MinLoCord MaxHiCord MaxSubmerge Is_Ogee
30,18,3,,50,50,,,0.95,0,1,1,,,
  3836.9  3860.1  3871.3  3894.5  3920.6  3937.9  3950.3  3978.8  3993.7  4039.2
  4072.3  4084.8  4110.0  4121.7  4127.4  4131.9  4155.8  4203.5  4220.8  4230.8
  4246.1  4253.3  4263.1  4330.4  4354.1  4396.3  4597.3  4642.9  4680.3  4761.6
  4804.1  4901.7  4932.1  4942.5  4959.1  4976.5  4976.5  5023.5  5023.5  5028.6
  5065.1  5095.5  5112.1  5130.7  5147.4  5176.0  5196.8  5214.0  5224.8  5236.9
  725.04  722.67  721.71  720.41  718.98  718.34  718.36  718.59  718.53  718.15
  717.84  717.71  717.69  718.63  719.06  719.16  718.67  715.38  712.41  710.32
  707.90  707.11  706.62  705.81  705.58  705.52  706.57  706.65  706.60  706.02
  706.29  707.05  708.49  708.89  709.04  708.82  708.82  708.63  708.63  708.61
  708.33  708.75  709.07  709.60  710.74  712.13  713.21  713.84  713.97  714.00
  677.46  677.46  677.46  677.46  677.46  677.46  677.46  677.46  677.46  677.46
  677.46  677.46  677.46  677.46  677.46  677.46  677.46  677.46  677.46  677.46
  677.46  677.46  677.46  677.46  677.46  677.46  677.46  677.46  677.46  677.46
  677.46  677.46  677.46  677.46  677.46  677.46  706.22  706.22  677.46  677.46
  677.46  677.46  677.46  677.46  677.46  677.46  677.46  677.46  677.46  677.46
  3836.9  3860.1  3871.3  3894.5  3920.6  3937.9  3950.3  3978.8  3993.7  4039.2
  4072.3  4084.8  4110.0  4121.7  4127.4  4131.9  4155.8  4203.5  4220.8  4230.8
  4246.1  4253.3  4263.1  4330.4  4354.1  4396.3  4597.3  4642.9  4680.3  4761.6
  4804.1  4901.7  4932.1  4942.5  4959.1  4976.5  4976.5  5023.5  5023.5  5028.6
  5065.1  5095.5  5112.1  5130.7  5147.4  5176.0  5196.8  5214.0  5224.8  5236.9
  725.04  722.67  721.71  720.41  718.98  718.34  718.36  718.59  718.53  718.15
  717.84  717.71  717.69  718.63  719.06  719.16  718.67  715.38  712.41  710.32
  707.90  707.11  706.62  705.81  705.58  705.52  706.57  706.65  706.60  706.02
  706.29  707.05  708.49  708.89  709.04  708.82  708.82  708.63  708.63  708.61
  708.33  708.75  709.07  709.60  710.74  712.13  713.21  713.84  713.97  714.00
  677.46  677.46  677.46  677.46  677.46  677.46  677.46  677.46  677.46  677.46
  677.46  677.46  677.46  677.46  677.46  677.46  677.46  677.46  677.46  677.46
  677.46  677.46  677.46  677.46  677.46  677.46  677.46  677.46  677.46  677.46
  677.46  677.46  677.46  677.46  677.46  677.46  706.22  706.22  677.46  677.46
  677.46  677.46  677.46  677.46  677.46  677.46  677.46  677.46  677.46  677.46
Abutment Skew #Up #Dn=,2,2
  4976.5  4980.0
  706.22  703.24
  4976.5  4980.0
  706.22  702.59
Abutment Skew #Up #Dn=,2,2
  5020.0  5023.5
  704.91  706.22
  5020.0  5023.5
  702.45  706.22
BR Coef=1,1,0,1.25,0,,,0.8,0,2,0,
WSPro=,,,, 1 ,,,, 0 ,,,, 0 ,,,,-1 ,-1 ,-1 , 0 , 0 , 0 , 0 , 0
BC Design=,,0,,0,,,,,,

Type RM Length L Ch R = 1,124141,918,918,918
BEGIN DESCRIPTION:
Murchison Rd (DC) ds
END DESCRIPTION:
XS GIS Cut Line= 6
      1529333.96       825298.53      1529407.12       824996.47
      1529196.28       824822.63      1528807.85       824800.11
      1528622.08       824541.15      1528354.71       824470.79
#Sta/Elev= 30
  3888.0  724.36  3962.4  717.95  4245.3  717.52  4287.1  714.37  4320.9  707.37
  4336.4  706.40  4470.2  705.49  4533.6  705.57  4581.6  705.51  4831.7  706.84
  4863.9  708.41  4923.5  706.58  4939.1  707.94  4969.2  706.00  4981.0  702.27
  4990.5  697.37  5009.5  697.37  5019.0  702.27  5048.9  707.77  5141.2  707.86
  5221.8  711.52  5245.4  715.04  5260.0  713.62  5299.0  718.01  5353.0  717.57
  5389.5  720.12  5416.2  720.03  5421.7  721.12  5458.3  721.92  5466.6  720.61
#Mann=6,-1,0
  3888.0    0.09       0  4470.2    0.14       0  4533.6    0.09       0
  4581.6    0.14       0  4981.0   0.045       0  5019.0    0.14       0
#XS Ineff=2,0
    0.00 4923.50  706.15 5076.50    0.00  708.52
Permanent Ineff=
       F       F
Bank Sta=4981,5019
XS Rating Curve= 0
Exp/Cntr=0.5,0.3

Type RM Length L Ch R = 1,123223,864,864,864
BEGIN DESCRIPTION:
Dutchman Creek 139.0
END DESCRIPTION:
XS GIS Cut Line= 5
      1529347.54       825304.84      1529420.71       824981.84
      1529459.63       824657.59      1529280.21       824047.55
      1529150.17       823931.26
#Sta/Elev= 30
  4428.4  724.64  4464.3  720.25  4531.4  716.95  4598.3  718.43  4691.0  717.00
  4775.3  717.00  4796.5  714.72  4813.3  714.00  4867.3  707.89  4881.4  704.85
  4905.9  705.53  4920.8  706.21  4979.8  703.92  4984.0  701.99  4985.7  696.99
  5014.3  696.99  5016.0  701.99  5035.0  704.62  5062.2  706.14  5240.8  704.83
  5335.4  705.35  5421.2  703.33  5468.2  704.92  5518.4  712.63  5536.0  713.94
  5593.2  715.29  5709.1  721.75  5793.5  725.48  5815.3  726.19  5896.5  726.36
#Mann=4,-1,0
  4428.4    0.09       0  4905.9    0.14       0  4984.0   0.045       0
  5016.0    0.06       0
Bank Sta=4984,5016
XS Rating Curve= 0
Exp/Cntr=0.3,0.1

Type RM Length L Ch R = 1,122359,757,757,757
BEGIN DESCRIPTION:
Dutchman Creek 138.0
END DESCRIPTION:
XS GIS Cut Line= 4
      1531026.02       825541.86      1530508.09       824613.37
      1529459.63       824164.94      1529219.64       823924.95
#Sta/Elev= 30
  3173.8  738.64  3267.9  735.86  3504.4  725.77  3562.5  721.08  3645.3  717.12
  3714.1  711.70  3836.9  708.87  3919.6  708.95  3972.7  708.56  3990.9  706.95
  4134.3  703.97  4538.2  704.88  4711.7  703.67  4927.0  704.68  4983.1  701.64
  4984.8  696.64  5015.2  696.64  5016.9  701.64  5037.8  704.96  5075.3  705.42
  5091.7  703.96  5284.4  704.28  5321.2  703.00  5390.9  706.58  5413.5  711.61
  5428.8  717.58  5450.4  719.36  5525.7  720.31  5645.8  724.55  5716.7  725.48
#Mann=4,-1,0
  3173.8    0.06       0  3919.6    0.14       0  4983.1   0.045       0
  5016.9    0.06       0
#XS Ineff=2,0
    0.00 3984.80  722.99               0
Permanent Ineff=
       F       F
Bank Sta=4983.1,5016.9
XS Rating Curve= 0
Exp/Cntr=0.3,0.1

Type RM Length L Ch R = 1,121602,891,891,891
BEGIN DESCRIPTION:
Dutchman Creek 137.0
END DESCRIPTION:
XS GIS Cut Line= 6
      1531752.33       824626.00      1531411.27       824209.15
      1530249.13       823994.41      1530047.02       823893.35
      1529554.37       823767.03      1529105.93       823861.77
#Sta/Elev= 30
  3114.6  761.43  3225.0  754.45  3338.6  740.25  3468.7  734.00  3540.7  732.89
  3574.0  728.57  3600.0  721.00  3635.5  715.51  3651.8  709.42  3663.8  707.70
  3754.9  705.22  3856.7  702.49  3982.0  702.20  4410.4  705.54  4973.7  704.99
  4983.1  701.33  4984.8  696.33  5015.2  696.33  5016.9  701.33  5058.6  704.76
  5209.9  703.45  5410.1  705.07  5441.7  703.57  5532.3  705.72  5541.5  705.98
  5578.9  714.77  5598.2  715.67  5722.1  717.76  5921.3  724.77  6027.9  725.57
#Mann=5,-1,0
  3114.6    0.14       0  3540.7    0.06       0  3754.9    0.14       0
  4983.1   0.045       0  5016.9    0.06       0
#XS Ineff=2,0
    0.00 4030.60  739.00               0
Permanent Ineff=
       F       F
Bank Sta=4983.1,5016.9
XS Rating Curve= 0
Exp/Cntr=0.3,0.1

Type RM Length L Ch R = 1,120711,790,790,790
BEGIN DESCRIPTION:
Dutchman Creek 136.0
END DESCRIPTION:
XS GIS Cut Line= 6
      1532030.22       823722.78      1531853.39       823369.12
      1530419.66       823337.54      1530135.44       823318.60
      1529889.12       823242.80      1529244.89       822421.72
#Sta/Elev= 30
  3058.6  748.07  3250.9  735.02  3411.6  728.29  3434.2  725.07  3492.4  707.29
  3527.7  705.82  3762.2  703.37  3801.9  701.35  4905.8  703.99  4964.0  703.18
  4970.8  701.18  4983.0  704.00  4983.1  700.96  4984.8  695.96  5015.2  695.96
  5016.9  700.96  5069.2  703.67  5155.8  704.50  5275.6  701.96  5368.2  709.58
  5565.1  707.58  5712.5  712.39  5915.4  719.38  5995.5  719.35  6055.4  716.86
  6075.3  711.02  6118.0  708.74  6259.3  717.66  6388.3  734.73  6474.3  741.05
#Mann=4,-1,0
  3058.6    0.14       0  4983.1   0.045       0  5016.9    0.14       0
  5712.5    0.06       0
#XS Ineff=2,0
    0.00 4000.00  727.33 5365.80    0.00  727.33
Permanent Ineff=
       F       F
Bank Sta=4983.1,5016.9
XS Rating Curve= 0
Exp/Cntr=0.3,0.1

Type RM Length L Ch R = 1,119921,1483,1483,1483
BEGIN DESCRIPTION:
Dutchman Creek 135.0
END DESCRIPTION:
XS GIS Cut Line= 5
      1531992.36       822964.91      1531670.23       822775.42
      1530659.67       822788.05      1529977.55       822598.57
      1529674.35       822200.63
#Sta/Elev= 30
  3134.8  752.91  3258.2  741.59  3390.7  721.94  3405.2  720.47  3441.7  721.36
  3456.1  717.90  3493.0  709.39  3519.8  706.27  3752.9  702.27  3791.9  703.33
  3951.1  701.01  4407.4  703.09  4522.3  700.23  4537.8  701.71  4948.2  703.16
  4979.4  701.65  4983.1  700.19  4984.8  695.19  5015.2  695.19  5016.9  700.19
  5018.4  703.27  5077.3  701.21  5156.2  709.01  5193.9  708.19  5249.4  702.92
  5311.6  703.30  5424.1  703.47  5483.6  711.81  5564.9  714.21  5727.4  725.26
#Mann=5,-1,0
  3134.8    0.14       0  3456.1    0.08       0  4983.1   0.045       0
  5016.9    0.08       0  5311.6    0.06       0
#XS Ineff=2,0
    0.00 3901.80  724.47 5179.10    0.00  724.47
Permanent Ineff=
       F       F
Bank Sta=4983.1,5016.9
XS Rating Curve= 0
Exp/Cntr=0.3,0.1

Type RM Length L Ch R = 1,118438,510,510,510
BEGIN DESCRIPTION:
Dutchman Creek 134.0
END DESCRIPTION:
XS GIS Cut Line= 4
      1531613.37       821966.98      1531190.21       822143.82
      1530665.82       822132.41      1529750.15       822099.61
#Sta/Elev= 30
  4474.8  734.39  4516.4  726.64  4585.9  715.77  4673.6  708.68  4722.6  703.05
  4802.0  699.58  4860.5  699.17  4902.5  701.02  4926.5  700.76  4955.5  698.55
  4983.1  698.34  4984.8  693.34  5015.2  693.34  5016.9  698.34  5018.0  701.46
  5047.9  701.03  5245.8  701.35  5319.4  700.93  5375.9  702.60  5443.9  701.29
  5491.3  703.97  5517.8  707.43  5572.8  708.53  5631.8  707.34  5727.3  707.61
  5791.6  709.05  5956.8  709.99  6046.1  711.63  6219.3  717.39  6374.2  727.07
#Mann=6,-1,0
  4474.8    0.14       0  4983.1   0.045       0  5016.9    0.14       0
  5047.9    0.06       0  5245.8    0.14       0  5631.8    0.06       0
Bank Sta=4983.1,5016.9
XS Rating Curve= 0
Exp/Cntr=0.3,0.1

Type RM Length L Ch R = 1,117928,634,634,634
BEGIN DESCRIPTION:
Dutchman Creek 133.0
END DESCRIPTION:
XS GIS Cut Line= 5
      1531619.65       821897.48      1531442.85       821828.02
      1531303.90       821834.34      1530261.76       821581.70
      1529863.84       821606.97
#Sta/Elev= 30
  4736.3  738.56  4774.8  733.50  4784.4  731.03  4826.2  724.30  4860.5  716.78
  4916.5  701.32  4930.6  700.00  4982.8  701.24  4983.1  697.89  4984.8  692.89
  5015.2  692.89  5016.9  697.89  5020.4  699.12  5044.4  701.02  5143.8  700.24
  5177.8  701.18  5260.7  700.11  5318.6  701.25  5452.8  700.50  5484.3  701.32
  5634.5  701.17  5919.2  699.71  6020.7  698.77  6236.8  702.15  6247.5  703.14
  6257.5  702.63  6326.6  707.90  6375.5  712.83  6464.4  717.76  6536.4  726.72
#Mann=5,-1,0
  4736.3    0.14       0  4983.1   0.045       0  5016.9    0.14       0
  5919.2    0.14       0  6326.6    0.06       0
#XS Ineff=2,0
       0                 5747.70    0.00  717.56
Permanent Ineff=
       F       F
Bank Sta=4983.1,5016.9
XS Rating Curve= 0
Exp/Cntr=0.3,0.1

Type RM Length L Ch R = 1,117294,457,457,457
BEGIN DESCRIPTION:
Dutchman Creek 132.0
END DESCRIPTION:
XS GIS Cut Line= 4
      1531842.04       821402.33      1531559.07       821356.85
      1531018.42       821089.05      1530907.27       820861.71
#Sta/Elev= 30
  4640.5  747.87  4693.7  743.72  4743.0  736.29  4802.4  724.10  4816.3  722.45
  4841.9  716.54  4867.1  709.13  4880.3  700.60  4904.1  699.20  4951.3  699.44
  4973.9  698.27  4983.1  697.34  4984.8  692.34  5015.2  692.34  5016.9  697.34
  5029.6  700.14  5093.8  698.57  5153.5  699.18  5167.6  700.30  5279.9  698.37
  5291.6  699.40  5405.6  699.83  5504.6  697.35  5519.4  697.81  5542.3  702.08
  5557.2  705.40  5595.6  709.81  5672.4  714.03  5734.5  717.24  5783.5  721.65
#Mann=6,-1,0
  4640.5    0.14       0  4973.9    0.06       0  4983.1   0.045       0
  5016.9    0.06       0  5542.3    0.14       0  5672.4    0.08       0
Bank Sta=4983.1,5016.9
XS Rating Curve= 0
Exp/Cntr=0.3,0.1

Type RM Length L Ch R = 1,116837,622,622,622
BEGIN DESCRIPTION:
Dutchman Creek 131.0
END DESCRIPTION:
XS GIS Cut Line= 5
      1531973.38       821230.52      1531670.23       821013.26
      1531362.01       820982.94      1531175.06       820866.73
      1530887.06       820816.20
#Sta/Elev= 30
  4447.6  749.70  4466.7  748.94  4504.2  743.40  4543.3  739.83  4604.4  726.40
  4653.6  719.42  4728.5  704.26  4756.3  701.00  4852.6  698.36  4957.5  699.38
  4970.4  700.51  4978.3  699.79  4983.1  696.94  4984.8  691.94  5015.2  691.94
  5016.9  696.94  5040.4  699.80  5076.8  698.83  5165.7  699.82  5263.7  698.05
  5319.6  698.73  5341.8  702.55  5345.4  705.06  5365.9  711.66  5388.0  714.98
  5418.9  717.81  5457.5  717.58  5497.9  716.82  5530.4  717.88  5642.8  725.75
#Mann=4,-1,0
  4447.6    0.14       0  4983.1   0.045       0  5016.9    0.14       0
  5457.5    0.08       0
Bank Sta=4983.1,5016.9
XS Rating Curve= 0
Exp/Cntr=0.3,0.1

Type RM Length L Ch R = 1,116215,473,473,473
BEGIN DESCRIPTION:
Dutchman Creek 130.0
END DESCRIPTION:
XS GIS Cut Line= 4
      1531836.94       820462.50      1531528.75       820427.14
      1531104.32       820523.14      1530775.89       820725.25
#Sta/Elev= 30
  4590.3  729.41  4735.4  723.26  4784.1  719.32  4864.8  709.19  4923.1  699.67
  4959.0  697.31  4980.1  697.74  4982.8  696.39  4984.5  691.39  5015.5  691.39
  5017.2  696.39  5019.6  699.48  5097.8  697.85  5121.6  698.46  5157.6  697.25
  5323.8  698.73  5337.9  697.06  5369.8  699.82  5403.9  700.75  5452.6  700.57
  5479.8  705.13  5494.8  705.79  5507.7  709.69  5522.3  712.48  5535.2  717.78
  5559.9  720.04  5588.5  723.08  5632.2  725.85  5671.7  725.99  5721.3  724.42
#Mann=5,-1,0
  4590.3    0.08       0  4864.8    0.14       0  4982.8   0.045       0
  5017.2    0.14       0  5559.9    0.08       0
Bank Sta=4982.8,5017.2
XS Rating Curve= 0
Exp/Cntr=0.3,0.1

Type RM Length L Ch R = 1,115742,1319,1319,1319
BEGIN DESCRIPTION:
Dutchman Creek 129.0
END DESCRIPTION:
XS GIS Cut Line= 4
      1531897.62       820351.36      1531629.81       820134.08
      1531432.75       820058.28      1530715.29       820209.86
#Sta/Elev= 30
  4366.9  728.15  4443.0  719.40  4495.5  716.01  4546.1  709.52  4691.2  703.30
  4723.9  699.93  4761.5  698.08  4844.0  698.21  4868.1  699.31  4929.2  698.12
  4951.0  698.86  4982.8  695.97  4984.5  690.97  5015.5  690.97  5017.2  695.97
  5046.4  699.13  5074.7  699.29  5119.9  698.14  5133.3  698.94  5147.3  697.80
  5169.9  698.44  5192.3  697.38  5291.2  699.54  5379.9  699.53  5391.4  699.47
  5409.6  697.40  5444.3  697.66  5491.1  702.35  5534.3  713.38  5656.2  727.47
#Mann=4,-1,0
  4366.9    0.08       0  4868.1    0.14       0  4982.8   0.045       0
  5017.2    0.14       0
Bank Sta=4982.8,5017.2
XS Rating Curve= 0
Exp/Cntr=0.3,0.1

Type RM Length L Ch R = 1,114423,1025,1025,1025
BEGIN DESCRIPTION:
Dutchman Creek 128.0
END DESCRIPTION:
XS GIS Cut Line= 4
      1532706.05       819563.11      1532433.20       819406.47
      1530775.89       819391.32      1530124.05       819244.78
#Sta/Elev= 30
  3446.4  740.12  3556.1  729.99  3660.0  724.04  3680.9  720.68  3733.2  712.30
  3743.9  704.91  3758.4  699.87  3815.0  695.58  4151.9  698.21  4675.5  698.19
  4951.7  698.30  4972.5  697.70  4982.8  694.46  4984.5  689.46  5015.5  689.46
  5017.2  694.46  5021.8  698.15  5032.3  698.46  5229.4  696.71  5406.2  698.25
  5468.7  695.73  5542.5  697.74  5607.4  696.29  5771.6  698.08  5872.4  701.98
  5893.9  700.11  5956.8  704.55  6044.6  727.69  6066.5  732.19  6086.5  732.73
#Mann=7,-1,0
  3446.4    0.08       0  3680.9    0.14       0  4675.5    0.14       0
  4951.7    0.06       0  4982.8   0.045       0  5017.2    0.06       0
  5229.4    0.14       0
#XS Ineff=2,0
    0.00 4157.70  717.36               0
Permanent Ineff=
       F       F
Bank Sta=4982.8,5017.2
XS Rating Curve= 0
Exp/Cntr=0.3,0.1

Type RM Length L Ch R = 1,113398,1384,1384,1384
BEGIN DESCRIPTION:
Dutchman Creek 127.0
END DESCRIPTION:
XS GIS Cut Line= 4
      1532867.70       818491.92      1531771.29       818643.50
      1530528.30       818461.60      1530058.41       818562.65
#Sta/Elev= 30
  3138.8  721.74  3224.9  718.98  3243.7  716.14  3257.9  710.20  3268.2  708.65
  3288.5  709.40  3352.7  700.35  3482.6  695.43  3812.1  693.82  3889.2  696.33
  4029.8  694.71  4196.2  696.62  4316.9  695.04  4424.5  696.81  4577.6  696.11
  4915.3  696.15  4967.5  698.05  4973.6  697.71  4982.8  692.87  4984.5  687.87
  5015.5  687.87  5017.2  692.87  5022.7  696.70  5055.4  697.21  5107.2  695.64
  5549.6  696.44  5641.2  700.57  5789.5  710.81  5914.9  714.16  5982.5  718.41
#Mann=5,-1,0
  3138.8    0.14       0  4577.6    0.06       0  4982.8   0.045       0
  5017.2    0.06       0  5789.5    0.06       0
#XS Ineff=2,0
    0.00 3965.70  709.37               0
Permanent Ineff=
       F       F
Bank Sta=4982.8,5017.2
XS Rating Curve= 0
Exp/Cntr=0.3,0.1

Type RM Length L Ch R = 1,112014,788,788,788
BEGIN DESCRIPTION:
Dutchman Creek 126.0
END DESCRIPTION:
XS GIS Cut Line= 3
      1532953.63       818188.75      1532130.03       818143.28
      1530811.25       817395.46
#Sta/Elev= 30
  3617.4  720.82  3658.7  720.06  3694.0  713.84  3749.0  710.25  4002.0  704.51
  4080.1  700.20  4100.3  696.73  4168.2  693.24  4285.0  695.85  4380.1  696.01
  4400.5  694.17  4608.2  695.27  4680.6  693.10  4811.2  695.25  4967.1  694.80
  4981.0  694.11  4982.8  690.98  4984.5  685.98  5015.5  685.98  5017.2  690.98
  5023.8  695.55  5608.7  693.91  5649.0  696.19  5716.6  695.14  5758.4  699.72
  5782.2  705.70  5801.7  710.66  5831.2  711.01  5864.4  714.87  5958.3  716.22
#Mann=6,-1,0
  3617.4    0.14       0  4967.1    0.06       0  4982.8   0.045       0
  5017.2    0.06       0  5608.7    0.14       0  5782.2    0.06       0
#XS Ineff=2,0
    0.00 4389.00  710.63               0
Permanent Ineff=
       F       F
Bank Sta=4982.8,5017.2
XS Rating Curve= 0
Exp/Cntr=0.3,0.1

Type RM Length L Ch R = 1,111226,488,488,488
BEGIN DESCRIPTION:
Dutchman Creek 125.0
END DESCRIPTION:
XS GIS Cut Line= 5
      1532679.57       817734.60      1532224.57       817657.60
      1531615.55       816838.57      1531536.43       816489.65
      1531328.53       816096.53
#Sta/Elev= 30
  3967.9  706.49  4037.2  704.35  4051.7  700.76  4084.2  701.31  4213.1  695.05
  4299.2  693.79  4312.1  691.13  4380.4  693.90  4709.2  694.74  4829.8  692.52
  4951.0  694.41  4976.7  691.93  4980.6  692.99  4982.8  689.91  4984.5  684.91
  5015.5  684.91  5017.2  689.91  5019.5  694.19  5023.7  694.44  5188.5  692.67
  5330.0  694.94  5612.4  695.27  5619.0  691.21  5624.3  691.20  5630.8  696.28
  5832.3  694.08  5892.1  698.28  6079.0  721.14  6192.0  735.33  6252.5  740.65
#Mann=7,-1,0
  3967.9    0.08       0  4951.0    0.06       0  4982.8   0.045       0
  5017.2    0.06       0  5612.4    0.05       0  5630.8    0.14       0
  6079.0    0.06       0
#XS Ineff=2,0
    0.00 4439.50  709.96               0
Permanent Ineff=
       F       F
Bank Sta=4982.8,5017.2
XS Rating Curve= 0
Exp/Cntr=0.3,0.1

Type RM Length L Ch R = 1,110738,607,607,607
BEGIN DESCRIPTION:
Dutchman Creek 124.0
END DESCRIPTION:
XS GIS Cut Line= 5
      1532718.77       817685.59      1532349.17       817343.99
      1532245.16       816805.90      1532052.36       815837.55
      1531828.34       815596.73
#Sta/Elev= 30
  4230.8  707.69  4371.5  702.25  4433.3  702.66  4476.2  697.98  4509.5  699.50
  4543.7  696.85  4930.1  690.54  4970.6  693.44  4982.7  694.01  4982.8  689.25
  4984.5  684.25  5015.5  684.25  5017.2  689.25  5029.1  693.31  5048.0  694.11
  5375.6  692.34  5450.4  694.54  5452.4  690.82  5455.9  690.94  5458.6  693.89
  5623.5  692.51  6253.9  696.00  6314.8  698.55  6386.2  708.02  6417.9  709.53
  6431.9  707.61  6458.3  716.62  6500.3  724.11  6549.7  730.89  6598.4  733.91
#Mann=7,-1,0
  4230.8    0.08       0  4970.6    0.06       0  4982.8   0.045       0
  5017.2    0.06       0  5375.6    0.14       0  5450.4    0.05       0
  5458.6    0.14       0
#XS Ineff=2,0
    0.00 4607.70  708.00 5900.00    0.00  708.00
Permanent Ineff=
       F       F
Bank Sta=4982.8,5017.2
XS Rating Curve= 0
Exp/Cntr=0.5,0.3

Type RM Length L Ch R = 1,110131,195,195,195
BEGIN DESCRIPTION:
Cana Rd (DC) us
END DESCRIPTION:
XS GIS Cut Line= 6
      1532752.37       817650.86      1532403.68       817373.74
      1532424.49       816450.11      1532291.56       816135.53
      1532279.17       815889.47      1532568.69       815079.33
#Sta/Elev= 30
  3741.9  709.75  3852.7  703.43  3975.0  703.33  4032.3  697.04  4086.6  699.40
  4189.1  694.80  4453.1  692.87  4541.0  694.79  4580.5  691.28  4599.0  695.21
  4700.7  696.79  4765.2  692.30  4797.3  694.73  4830.5  692.67  4902.6  694.17
  4924.2  690.19  4963.9  693.62  4981.0  690.32  4987.5  683.42  5012.5  683.42
  5019.0  690.32  5240.0  694.68  5381.2  692.34  5452.8  696.28  5993.4  696.32
  6108.2  700.68  6251.9  715.73  6423.5  719.71  6498.3  725.56  6590.5  725.60
#Mann=5,-1,0
  3741.9    0.08       0  4453.1    0.06       0  4830.5    0.14       0
  4981.0   0.045       0  5019.0    0.14       0
#XS Ineff=2,0
    0.00 4896.00  697.24 5104.00    0.00  699.82
Permanent Ineff=
       F       F
Bank Sta=4981,5019
XS Rating Curve= 0
Exp/Cntr=0.5,0.3

Type RM Length L Ch R =3,110067,,,
BEGIN DESCRIPTION:
Cana Rd (DC) tor
Structure ID: LDS_DC_09-1
Approximate Survey Structure
END DESCRIPTION:
Bridge Culvert--1,0,-1,-1,0
Deck Dist Width WeirC Skew NumUp NumDn MinLoCord MaxHiCord MaxSubmerge Is_Ogee
29,26,3,,35,35,,,0.95,0,1,1,,,
  3737.9  3857.0  3865.5  3911.1  3940.6  4173.4  4249.3  4357.4  4476.2  4545.8
  4677.1  4710.8  4781.3  4925.0  4925.0  5075.0  5075.0  5091.7  5171.7  5210.7
  5241.2  5299.3  5444.6  5496.7  5546.2  5603.3  5651.5  5698.6  5786.7  5837.0
  5906.0  5959.0  6005.6  6165.3  6819.6
  722.11  712.81  711.75  708.23  706.68  701.55  699.55  698.31  697.22  697.42
  698.45  698.56  699.99  701.92  701.92  701.92  701.92  701.85  700.43  699.39
  699.30  699.36  704.49  706.85  709.29  710.57  711.31  710.66  706.86  705.51
  704.82  704.85  706.29  713.10  736.74
  663.42  663.42  663.42  663.42  663.42  663.42  663.42  663.42  663.42  663.42
  663.42  663.42  663.42  663.42  698.22  698.22  663.42  663.42  663.42  663.42
  663.42  663.42  663.42  663.42  663.42  663.42  663.42  663.42  663.42  663.42
  663.42  663.42  663.42  663.42  663.42
  3737.9  3857.0  3865.5  3911.1  3940.6  4173.4  4249.3  4357.4  4476.2  4545.8
  4677.1  4710.8  4781.3  4925.0  4925.0  5075.0  5075.0  5091.7  5171.7  5210.7
  5241.2  5299.3  5444.6  5496.7  5546.2  5603.3  5651.5  5698.6  5786.7  5837.0
  5906.0  5959.0  6005.6  6165.3  6819.6
  722.11  712.81  711.75  708.23  706.68  701.55  699.55  698.31  697.22  697.42
  698.45  698.56  699.99  701.92  701.92  701.92  701.92  701.85  700.43  699.39
  699.30  699.36  704.49  706.85  709.29  710.57  711.31  710.66  706.86  705.51
  704.82  704.85  706.29  713.10  736.74
  663.42  663.42  663.42  663.42  663.42  663.42  663.42  663.42  663.42  663.42
  663.42  663.42  663.42  663.42  698.22  698.22  663.42  663.42  663.42  663.42
  663.42  663.42  663.42  663.42  663.42  663.42  663.42  663.42  663.42  663.42
  663.42  663.42  663.42  663.42  663.42
Pier Skew, UpSta & Num, DnSta & Num=,4943.8,2,4943.8,2,0,0,0,0,0
       1       1
  692.94  698.22
       1       1
  693.39  698.22
Pier Skew, UpSta & Num, DnSta & Num=,4981.3,2,4981.3,2,0,0,0,0,0
       1       1
  690.00  698.22
       1       1
  689.75  698.22
Pier Skew, UpSta & Num, DnSta & Num=,5018.8,2,5018.8,2,0,0,0,0,0
       1       1
  690.11  698.22
       1       1
  689.86  698.22
Pier Skew, UpSta & Num, DnSta & Num=,5056.3,2,5056.3,2,0,0,0,0,0
       1       1
  695.50  698.22
       1       1
  694.38  698.22
Abutment Skew #Up #Dn=,2,2
  4925.0  4926.5
  698.22  690.51
  4925.0  4926.5
  698.22  692.72
Abutment Skew #Up #Dn=,2,2
  5073.5  5075.0
  695.58  698.22
  5073.5  5075.0
  694.20  698.22
BR Coef=1,1,0,1.25,0,,,0.8,0,2,0,
WSPro=,,,, 1 ,,,, 0 ,,,, 0 ,,,,-1 ,-1 ,-1 , 0 , 0 , 0 , 0 , 0
BC Design=,,0,,0,,,,,,

Type RM Length L Ch R = 1,109936,1073,1073,1073
BEGIN DESCRIPTION:
Cana Rd (DC) ds
END DESCRIPTION:
XS GIS Cut Line= 5
      1532815.13       817503.06      1532564.22       817261.11
      1532613.50       816638.37      1532662.78       815979.79
      1532941.34       814878.34
#Sta/Elev= 30
  3951.6  716.38  4006.4  710.63  4108.3  707.36  4132.7  702.07  4250.6  695.68
  4423.4  693.24  4648.5  691.93  4845.2  693.58  4899.5  691.65  4963.5  693.94
  4981.0  690.07  4987.5  683.17  5012.5  683.17  5019.0  690.07  5031.4  694.03
  5119.7  694.62  5520.1  691.82  5765.9  692.31  5886.3  695.68  5942.6  695.45
  6080.2  700.10  6162.9  708.09  6260.5  721.64  6271.5  724.94  6302.2  727.02
  6332.9  731.71  6460.6  745.25  6596.9  757.12  6671.2  760.92  6721.4  759.55
#Mann=5,-1,0
  3951.6    0.08       0  4423.4    0.06       0  4845.2    0.14       0
  4981.0   0.045       0  5019.0    0.14       0
#XS Ineff=2,0
    0.00 4810.00  697.59 5190.00    0.00  699.49
Permanent Ineff=
       F       F
Bank Sta=4981,5019
XS Rating Curve= 0
Exp/Cntr=0.5,0.3

Type RM Length L Ch R = 1,108863,853,853,853
BEGIN DESCRIPTION:
Dutchman Creek 123.0
END DESCRIPTION:
XS GIS Cut Line= 5
      1533736.61       817517.55      1533715.61       816831.57
      1533526.60       815879.55      1533260.60       815389.53
      1533113.60       815151.54
#Sta/Elev= 30
  3831.7  737.29  3893.2  734.88  4038.4  719.26  4099.7  714.30  4329.0  706.03
  4363.7  703.67  4469.6  692.23  4571.9  690.96  4614.9  691.98  4780.8  691.06
  4946.9  692.99  4959.4  692.74  4980.9  687.54  4982.6  682.54  5017.4  682.54
  5019.1  687.54  5037.6  693.48  5123.7  691.87  5363.7  692.31  5666.5  689.78
  5686.8  691.13  5730.6  689.55  6047.7  691.52  6070.6  693.96  6086.1  698.54
  6167.2  737.16  6192.4  743.90  6228.5  746.01  6277.5  742.12  6325.9  741.34
#Mann=5,-1,0
  3831.7    0.14       0  4571.9    0.06       0  4946.9    0.14       0
  4980.9   0.045       0  5019.1    0.14       0
Bank Sta=4980.9,5019.1
XS Rating Curve= 0
Exp/Cntr=0.3,0.1

Type RM Length L Ch R = 1,108010,564,564,564
BEGIN DESCRIPTION:
Dutchman Creek 122.0
END DESCRIPTION:
XS GIS Cut Line= 3
      1534529.86       816321.39      1534337.87       816152.67
      1534151.67       814890.01
#Sta/Elev= 30
  4851.7  718.97  4924.3  721.42  4939.6  719.81  4947.1  717.30  4961.1  708.66
  4971.1  705.14  4980.9  687.04  4982.6  682.04  5017.4  682.04  5019.1  687.04
  5020.2  689.72  5027.7  690.38  5102.0  692.51  5236.5  690.20  5419.0  691.85
  5512.7  690.19  5562.8  691.27  5691.9  690.91  5800.3  690.76  5910.0  688.77
  5972.6  689.65  5995.0  688.59  6056.2  690.44  6084.5  693.84  6128.5  705.12
  6229.7  745.36  6281.2  762.88  6308.1  768.20  6322.0  769.43  6383.6  769.67
#Mann=4,-1,0
  4851.7    0.08       0  4980.9   0.045       0  5019.1    0.08       0
  5691.9    0.14       0
Bank Sta=4980.9,5019.1
XS Rating Curve= 0
Exp/Cntr=0.3,0.1

Type RM Length L Ch R = 1,107446,969,969,969
BEGIN DESCRIPTION:
Dutchman Creek 121.0
END DESCRIPTION:
XS GIS Cut Line= 5
      1534797.56       816379.62      1534803.38       816187.58
      1534774.29       815780.26      1534832.48       815367.12
      1535175.76       815000.57
#Sta/Elev= 30
  4716.4  715.50  4739.8  715.51  4753.3  714.67  4799.1  703.88  4867.7  692.76
  4893.5  691.33  4973.0  691.25  4980.9  686.71  4982.6  681.71  5017.4  681.71
  5019.1  686.71  5037.2  691.06  5058.9  691.70  5207.0  690.67  5330.3  691.08
  5380.6  689.41  5424.5  690.32  5531.7  690.12  5680.3  688.76  5829.3  689.25
  5839.0  688.50  5907.5  689.99  5966.4  692.79  5997.7  696.41  6047.8  704.47
  6081.2  712.37  6154.1  737.36  6189.4  747.38  6223.7  752.26  6236.3  753.13
#Mann=4,-1,0
  4716.4    0.08       0  4980.9   0.045       0  5019.1    0.08       0
  5531.7    0.14       0
Bank Sta=4980.9,5019.1
XS Rating Curve= 0
Exp/Cntr=0.3,0.1

Type RM Length L Ch R = 1,106477,592,592,592
BEGIN DESCRIPTION:
Dutchman Creek 120.0
END DESCRIPTION:
XS GIS Cut Line= 4
      1535643.09       817372.73      1535643.09       816347.19
      1535492.27       815653.45      1535534.50       815418.19
#Sta/Elev= 30
  3513.0  718.64  3667.8  708.14  3867.0  701.26  4140.9  700.17  4323.6  697.95
  4475.1  699.05  4611.2  697.89  4707.3  699.49  4754.9  695.45  4794.0  688.89
  4867.6  690.19  4974.9  690.62  4980.9  686.14  4982.6  681.14  5017.4  681.14
  5019.1  686.14  5023.8  690.67  5050.8  689.10  5066.5  690.66  5140.2  689.80
  5226.3  690.72  5248.5  692.04  5281.2  695.95  5309.1  701.03  5364.7  713.33
  5407.3  724.36  5421.7  726.13  5443.8  731.17  5457.3  732.56  5487.5  738.89
#Mann=4,-1,0
  3513.0    0.08       0  4867.6    0.14       0  4980.9   0.045       0
  5019.1    0.14       0
Bank Sta=4980.9,5019.1
XS Rating Curve= 0
Exp/Cntr=0.3,0.1

Type RM Length L Ch R = 1,105885,1183,1183,1183
BEGIN DESCRIPTION:
Dutchman Creek 119.0
END DESCRIPTION:
XS GIS Cut Line= 6
      1536562.80       817025.62      1536157.54       816465.79
      1536157.54       816114.46      1536053.30       815724.51
      1535988.60       815521.38      1535737.86       815278.73
#Sta/Elev= 30
  3641.9  718.26  3674.6  710.80  3713.0  709.43  3738.7  712.60  3753.9  709.71
  3803.5  706.30  3974.6  699.08  4100.6  695.34  4245.6  695.04  4466.1  692.24
  4599.5  692.68  4699.6  694.62  4767.1  688.70  4843.5  687.22  4865.7  688.85
  4960.6  690.56  4976.2  689.74  4980.9  685.79  4982.6  680.79  5017.4  680.79
  5019.1  685.79  5029.3  689.91  5089.1  691.45  5134.8  696.18  5171.1  696.54
  5216.6  700.94  5301.2  712.19  5573.1  758.20  5614.4  763.17  5650.1  764.23
#Mann=6,-1,0
  3641.9    0.08       0  3974.6    0.14       0  4245.6    0.08       0
  4699.6    0.14       0  4980.9   0.045       0  5019.1    0.14       0
Bank Sta=4980.9,5019.1
XS Rating Curve= 0
Exp/Cntr=0.3,0.1

Type RM Length L Ch R = 1,104702,948,948,948
BEGIN DESCRIPTION:
Dutchman Creek 118.0
END DESCRIPTION:
XS GIS Cut Line= 5
      1537258.96       817252.42      1537305.51       816711.28
      1536682.89       815483.50      1536595.60       815262.38
      1536444.32       815018.01
#Sta/Elev= 30
  3631.8  740.74  3708.7  735.12  3731.9  731.07  3740.6  725.28  3749.6  726.08
  3784.9  719.00  3853.4  712.64  3876.2  707.01  3892.0  707.49  3953.0  701.78
  4127.3  691.96  4205.4  688.22  4278.9  688.51  4971.7  690.27  4980.4  689.14
  4980.9  685.09  4982.6  680.09  5017.4  680.09  5019.1  685.09  5019.3  690.49
  5333.2  687.73  5413.5  689.41  5476.8  687.92  5558.2  692.64  5649.1  690.68
  5773.5  698.72  5933.5  716.56  5995.8  722.28  6015.2  721.47  6076.7  729.53
#Mann=5,-1,0
  3631.8    0.08       0  4127.3    0.14       0  4278.9    0.08       0
  4980.9   0.045       0  5019.1    0.08       0
Bank Sta=4980.9,5019.1
XS Rating Curve= 0
Exp/Cntr=0.3,0.1

Type RM Length L Ch R = 1,103754,962,962,962
BEGIN DESCRIPTION:
Dutchman Creek 117.0
END DESCRIPTION:
XS GIS Cut Line= 5
      1538224.89       816914.95      1538003.77       816513.44
      1537672.10       815879.18      1537334.60       815169.28
      1537375.34       814389.50
#Sta/Elev= 30
  3783.4  711.06  3899.0  702.18  4170.5  694.21  4239.5  694.63  4312.6  688.45
  4387.8  686.97  4570.0  687.06  4585.9  688.27  4682.9  687.24  4827.3  689.33
  4866.5  688.32  4965.1  689.30  4980.9  684.54  4982.6  679.54  5017.4  679.54
  5019.1  684.54  5027.9  689.44  5347.1  687.66  5642.8  689.61  5933.5  688.17
  6028.6  688.86  6054.3  690.37  6076.6  689.42  6191.0  693.04  6203.4  696.34
  6216.6  702.09  6271.0  711.15  6354.0  717.33  6432.3  726.73  6524.4  735.15
#Mann=6,-1,0
  3783.4    0.08       0  4170.5    0.14       0  4866.5    0.08       0
  4980.9   0.045       0  5019.1    0.08       0  5642.8    0.14       0
#XS Ineff=2,0
       0                 5773.60    0.00  715.24
Permanent Ineff=
       F       F
Bank Sta=4980.9,5019.1
XS Rating Curve= 0
Exp/Cntr=0.3,0.1

Type RM Length L Ch R = 1,102792,1191,1191,1191
BEGIN DESCRIPTION:
Dutchman Creek 116.0
END DESCRIPTION:
XS GIS Cut Line= 4
      1538481.11       816818.59      1538181.88       816139.25
      1538278.93       815742.97      1537478.30       814400.49
#Sta/Elev= 30
  3456.1  719.37  3502.5  713.77  3622.3  704.53  3789.8  698.19  4015.7  695.56
  4217.1  697.06  4342.2  692.32  4531.9  691.27  4652.2  691.04  4684.1  687.96
  4689.2  685.05  4696.5  684.27  4726.7  684.27  4766.6  688.29  4871.1  688.84
  4963.4  688.03  4980.9  683.97  4982.6  678.97  5017.4  678.97  5019.1  683.97
  5045.1  692.35  5066.4  693.12  5150.7  687.35  5424.0  688.40  5447.1  686.70
  5710.0  691.29  5797.6  695.23  5949.7  707.05  6034.7  718.92  6169.5  729.44
#Mann=4,-1,0
  3456.1    0.08       0  4531.9    0.14       0  4980.9   0.045       0
  5019.1    0.14       0
#XS Ineff=2,0
       0                 5559.00    0.00  711.87
Permanent Ineff=
       F       F
Bank Sta=4980.9,5019.1
XS Rating Curve= 0
Exp/Cntr=0.3,0.1

Type RM Length L Ch R = 1,101601,1956,1956,1956
BEGIN DESCRIPTION:
Dutchman Creek 115.0
END DESCRIPTION:
XS GIS Cut Line= 4
      1539283.37       816689.19      1539153.98       816114.99
      1538749.61       814554.14      1538555.52       814101.26
#Sta/Elev= 30
  3799.3  714.63  3842.7  709.50  3958.7  702.97  4174.2  696.63  4209.4  696.43
  4349.3  688.59  4438.9  686.48  4613.9  685.30  4959.2  687.77  4976.4  687.64
  4980.9  683.27  4982.6  678.27  5017.4  678.27  5019.1  683.27  5035.6  687.74
  5095.3  687.27  5106.2  685.92  5142.0  687.38  5322.2  687.20  5387.5  685.59
  5448.0  687.29  5506.2  685.86  5542.9  686.95  5636.3  685.35  5839.9  685.67
  5999.4  689.20  6124.8  695.73  6189.7  696.75  6276.4  701.12  6493.0  718.80
#Mann=5,-1,0
  3799.3    0.08       0  4174.2    0.14       0  4980.9   0.045       0
  5019.1    0.14       0  5839.9    0.08       0
#XS Ineff=2,0
       0                 5737.80    0.00  705.68
Permanent Ineff=
       F       F
Bank Sta=4980.9,5019.1
XS Rating Curve= 0
Exp/Cntr=0.3,0.1

Type RM Length L Ch R = 1,99645,1276,1276,1276
BEGIN DESCRIPTION:
Dutchman Creek 114.0
END DESCRIPTION:
XS GIS Cut Line= 4
      1540447.70       815663.88      1540209.13       815308.93
      1539010.44       814249.89      1538690.42       813993.88
#Sta/Elev= 30
  4650.1  733.07  4714.0  723.77  4724.0  723.78  4787.3  713.35  4802.2  713.00
  4871.9  701.59  4953.3  693.78  4980.2  687.19  4980.9  681.94  4982.6  676.94
  5017.4  676.94  5019.1  681.94  5028.1  685.54  5066.9  685.97  5210.6  686.02
  5230.1  684.15  5254.1  685.45  5320.7  682.96  5394.0  685.64  5446.5  684.16
  5621.0  686.17  5912.1  684.27  6167.7  686.25  6677.7  685.18  6689.7  685.13
  6694.8  687.29  6727.0  691.53  6801.9  695.10  6921.9  706.04  7087.1  723.41
#Mann=5,-1,0
  4650.1    0.05       0  4953.3    0.14       0  4980.9   0.045       0
  5019.1    0.14       0  6677.7    0.08       0
#XS Ineff=2,0
       0                 6173.40    0.00  714.20
Permanent Ineff=
       F       F
Bank Sta=4980.9,5019.1
XS Rating Curve= 0
Exp/Cntr=0.3,0.1

Type RM Length L Ch R = 1,98369,660,660,660
BEGIN DESCRIPTION:
Dutchman Creek 113.0
END DESCRIPTION:
XS GIS Cut Line= 5
      1540983.07       815192.59      1540523.35       814418.64
      1540389.52       814278.99      1539842.54       813470.16
      1539854.18       813173.42
#Sta/Elev= 30
  3974.2  719.24  4110.9  703.83  4187.9  698.14  4286.7  694.29  4433.8  691.99
  4466.7  693.40  4566.5  686.50  4664.5  685.69  4697.1  682.89  4764.7  682.45
  4847.9  684.22  4890.4  682.92  4945.3  684.92  4966.7  684.31  4980.9  681.27
  4982.6  676.27  5017.4  676.27  5019.1  681.27  5029.9  683.80  5110.8  682.22
  5146.8  683.63  5186.4  681.09  5207.1  683.43  5299.0  684.39  5601.0  685.09
  5951.4  683.37  6018.8  685.08  6054.2  702.72  6281.2  724.66  6341.2  732.09
#Mann=4,-1,0
  3974.2    0.05       0  4664.5    0.14       0  4980.9   0.045       0
  5019.1    0.14       0
#XS Ineff=2,0
       0                 5577.00    0.00  709.26
Permanent Ineff=
       F       F
Bank Sta=4980.9,5019.1
XS Rating Curve= 0
Exp/Cntr=0.3,0.1

Type RM Length L Ch R = 1,97709,825,825,825
BEGIN DESCRIPTION:
Dutchman Creek 112.0
END DESCRIPTION:
XS GIS Cut Line= 5
      1541058.69       815221.67      1541052.87       814599.03
      1541017.96       814343.00      1540878.31       813662.19
      1540959.78       813289.75
#Sta/Elev= 30
  3824.0  724.34  3857.3  720.77  3928.2  719.59  3970.7  712.44  3993.0  711.62
  4041.7  705.16  4149.4  698.85  4214.5  692.32  4309.0  691.18  4374.7  695.83
  4460.5  695.60  4633.1  687.24  4692.7  689.14  4722.5  684.66  4732.2  682.51
  4778.0  681.78  4963.9  684.58  4980.0  682.90  4980.9  681.06  4982.6  676.06
  5017.4  676.06  5019.1  681.06  5022.5  684.20  5038.4  683.34  5205.6  681.46
  5300.2  683.49  5462.8  690.35  5547.5  696.60  5726.1  707.13  5781.3  710.36
#Mann=8,-1,0
  3824.0    0.05       0  4722.5    0.14       0  4980.9   0.045       0
  5019.1    0.14       0  5038.4    0.06       0  5300.2    0.14       0
  5547.5    0.06       0  5726.1    0.14       0
Bank Sta=4980.9,5019.1
XS Rating Curve= 0
Exp/Cntr=0.3,0.1

Type RM Length L Ch R = 1,96884,1043,1043,1043
BEGIN DESCRIPTION:
Dutchman Creek 111.0
END DESCRIPTION:
XS GIS Cut Line= 4
      1542653.07       815204.20      1541937.34       814040.41
      1541384.55       813807.66      1541023.78       813272.33
#Sta/Elev= 30
  3345.3  705.36  3522.4  702.43  3673.3  698.46  3753.5  694.95  3879.1  692.26
  4329.3  688.50  4353.4  689.23  4458.2  688.56  4518.4  689.89  4532.4  688.97
  4712.1  694.06  4757.3  692.24  4897.9  691.34  4972.6  683.81  4979.3  680.52
  4981.0  675.52  5019.0  675.52  5020.7  680.52  5086.8  682.62  5335.3  681.95
  5570.0  683.69  5649.9  682.74  5687.1  682.43  5737.0  686.40  5752.1  690.79
  5772.6  693.89  5779.3  696.74  5857.7  707.33  5919.7  712.32  5956.9  713.89
#Mann=6,-1,0
  3345.3    0.06       0  4353.4    0.05       0  4757.3    0.06       0
  4979.3   0.045       0  5020.7    0.06       0  5649.9    0.14       0
#XS Ineff=2,0
    0.00 4717.20  701.69               0
Permanent Ineff=
       F       F
Bank Sta=4979.3,5020.7
XS Rating Curve= 0
Exp/Cntr=0.3,0.1

Type RM Length L Ch R = 1,95841,804,804,804
BEGIN DESCRIPTION:
Dutchman Creek 110.0
END DESCRIPTION:
XS GIS Cut Line= 5
      1543554.98       814354.60      1543403.70       814033.43
      1543147.67       813551.63      1541867.52       813204.82
      1541582.39       812649.69
#Sta/Elev= 30
  3277.9  707.06  3507.1  701.01  3795.2  697.24  4166.9  689.31  4216.8  686.28
  4299.9  683.51  4474.7  683.55  4533.5  684.94  4650.7  683.64  4736.0  684.57
  4781.3  683.92  4831.8  680.66  4955.6  681.45  4979.3  679.83  4981.0  674.83
  5019.0  674.83  5020.7  679.83  5027.7  682.93  5049.5  681.41  5133.0  680.68
  5568.8  682.26  5790.3  686.63  5849.5  689.08  5872.7  691.16  5920.7  697.72
  5956.2  704.14  5991.8  717.86  6041.3  729.68  6096.3  736.06  6128.9  738.29
#Mann=4,-1,0
  3277.9    0.06       0  4979.3   0.045       0  5020.7    0.06       0
  5568.8    0.14       0
#XS Ineff=2,0
    0.00 4319.80  710.49               0
Permanent Ineff=
       F       F
Bank Sta=4979.3,5020.7
XS Rating Curve= 0
Exp/Cntr=0.3,0.1

Type RM Length L Ch R = 1,95037,552,552,552
BEGIN DESCRIPTION:
Dutchman Creek 109.0
END DESCRIPTION:
XS GIS Cut Line= 6
      1543953.00       813209.47      1543496.81       813121.03
      1543198.88       813144.30      1542873.02       812981.37
      1542225.96       812865.00      1542039.74       812622.89
#Sta/Elev= 30
  3124.0  700.93  3190.5  698.37  3504.3  692.47  3735.1  689.63  3767.7  688.40
  3805.2  683.75  3829.1  682.51  3849.0  679.06  3876.1  679.54  3892.5  677.37
  3896.9  679.85  3919.6  678.67  3932.6  680.38  3943.1  679.77  4033.3  679.00
  4090.3  678.67  4192.3  681.74  4247.9  680.05  4401.8  681.66  4620.1  681.25
  4632.9  682.34  4919.2  681.14  4969.0  680.57  4979.3  679.17  4981.0  674.17
  5019.0  674.17  5020.7  679.17  5070.3  696.32  5205.8  718.75  5228.6  720.63
#Mann=6,-1,0
  3124.0    0.08       0  3735.1    0.14       0  3943.1    0.06       0
  4033.3    0.14       0  4979.3   0.045       0  5020.7    0.14       0
Bank Sta=4979.3,5020.7
XS Rating Curve= 0
Exp/Cntr=0.3,0.1

Type RM Length L Ch R = 1,94485,1167,1167,1167
BEGIN DESCRIPTION:
Dutchman Creek 108.0
END DESCRIPTION:
XS GIS Cut Line= 4
      1543942.06       813186.79      1543493.35       813074.62
      1542994.05       812837.07      1542286.48       812259.84
#Sta/Elev= 30
  3197.6  700.26  3565.2  693.53  3723.1  692.53  3809.0  689.50  3869.2  686.80
  3928.6  686.42  3977.7  683.04  4000.7  678.94  4027.9  677.30  4148.5  679.74
  4232.5  677.49  4277.8  679.43  4626.2  681.56  4690.0  681.18  4714.7  678.85
  4798.7  681.59  4902.0  681.29  4930.1  679.75  4970.5  681.40  4979.3  678.71
  4981.0  673.71  5019.0  673.71  5020.7  678.71  5022.9  680.75  5040.3  681.95
  5045.7  684.10  5065.3  699.47  5082.0  708.04  5103.5  712.92  5126.2  713.99
#Mann=4,-1,0
  3197.6    0.08       0  3809.0    0.14       0  4979.3   0.045       0
  5020.7    0.14       0
Bank Sta=4979.3,5020.7
XS Rating Curve= 0
Exp/Cntr=0.3,0.1

Type RM Length L Ch R = 1,93318,878,878,878
BEGIN DESCRIPTION:
Dutchman Creek 107.0
END DESCRIPTION:
XS GIS Cut Line= 3
      1543974.16       813162.77      1543517.39       813026.54
      1542611.99       812145.17
#Sta/Elev= 30
  4101.7  703.92  4139.6  700.31  4156.6  699.75  4314.9  697.85  4381.6  695.72
  4520.1  693.44  4636.5  692.55  4787.4  687.95  4887.3  684.98  4928.5  682.35
  4942.9  678.79  4979.3  677.75  4981.0  672.75  5019.0  672.75  5020.7  677.75
  5028.4  680.59  5033.5  679.33  5070.4  680.69  5142.4  679.59  5266.6  681.38
  5289.4  680.52  5430.2  681.22  5457.9  681.14  5477.8  679.76  5497.0  681.87
  5537.0  689.64  5556.0  691.92  5618.9  695.44  5727.6  704.83  5841.9  708.00
#Mann=4,-1,0
  4101.7    0.08       0  4787.4    0.14       0  4979.3   0.045       0
  5020.7    0.14       0
Bank Sta=4979.3,5020.7
XS Rating Curve= 0
Exp/Cntr=0.3,0.1

Type RM Length L Ch R = 1,92440,1171,1171,1171
BEGIN DESCRIPTION:
Dutchman Creek 106.0
END DESCRIPTION:
XS GIS Cut Line= 6
      1544055.44       812608.99      1543822.66       812315.69
      1543673.70       812068.97      1543487.50       811975.87
      1542714.75       811775.70      1542407.53       811715.19
#Sta/Elev= 30
  4271.9  704.18  4671.8  689.33  4710.0  686.09  4738.6  682.28  4746.8  679.22
  4762.7  678.45  4896.5  680.12  4912.2  676.50  4917.4  680.14  4968.2  678.25
  4979.3  677.02  4981.0  672.02  5019.0  672.02  5020.7  677.02  5023.7  679.77
  5030.6  680.05  5494.4  679.78  5513.6  681.17  5549.0  677.42  5566.0  678.28
  5595.9  679.72  5783.1  680.57  5841.1  682.64  5872.7  681.33  5895.6  684.11
  5996.6  687.29  6086.6  694.07  6132.7  698.87  6179.9  706.74  6254.1  709.05
#Mann=6,-1,0
  4271.9    0.14       0  4968.2    0.06       0  4979.3   0.045       0
  5020.7    0.06       0  5494.4    0.14       0  5566.0    0.06       0
#XS Ineff=2,0
       0                 5594.10    0.00  704.00
Permanent Ineff=
       F       F
Bank Sta=4979.3,5020.7
XS Rating Curve= 0
Exp/Cntr=0.3,0.1

Type RM Length L Ch R = 1,91269,557,557,557
BEGIN DESCRIPTION:
Dutchman Creek 105.0
END DESCRIPTION:
XS GIS Cut Line= 5
      1544539.59       811552.27      1544371.97       811487.08
      1543925.08       811477.77      1543091.81       811040.19
      1542868.37       810863.30
#Sta/Elev= 30
  4732.1  708.12  4791.2  705.53  4867.3  700.17  4909.9  694.92  4913.4  693.53
  4950.3  679.20  4971.5  679.14  4979.3  676.05  4981.0  671.05  5019.0  671.05
  5020.7  676.05  5022.6  678.72  5122.2  677.45  5165.5  678.15  5189.3  679.27
  5405.7  678.14  5493.2  679.50  5798.3  677.01  6073.8  677.37  6101.0  676.32
  6170.8  677.67  6238.9  677.34  6276.1  678.66  6302.8  681.58  6323.3  685.09
  6345.8  691.52  6410.1  706.47  6424.4  708.24  6475.5  712.93  6585.1  716.71
#Mann=5,-1,0
  4732.1    0.06       0  4913.4    0.14       0  4979.3   0.045       0
  5020.7    0.14       0  5165.5    0.06       0
#XS Ineff=2,0
       0                 5975.00    0.00  708.00
Permanent Ineff=
       F       F
Bank Sta=4979.3,5020.7
XS Rating Curve= 0
Exp/Cntr=0.3,0.1

Type RM Length L Ch R = 1,90712,1027,1027,1027
BEGIN DESCRIPTION:
Dutchman Creek 104.0
END DESCRIPTION:
XS GIS Cut Line= 4
      1544759.31       811186.81      1544454.87       810994.53
      1543910.01       811018.57      1542796.24       810754.15
#Sta/Elev= 30
  4411.0  708.22  4512.3  705.99  4584.8  702.17  4806.0  695.74  4877.2  691.26
  4948.3  684.22  4975.0  679.70  4979.3  675.60  4981.0  670.60  5019.0  670.60
  5020.7  675.60  5024.5  678.54  5034.2  678.65  5131.8  677.07  5217.9  677.99
  5269.2  676.71  5309.3  678.42  5463.5  677.89  5491.9  675.18  5509.3  676.96
  5538.5  677.53  5988.0  677.86  6038.6  676.96  6104.0  681.85  6132.4  687.38
  6178.1  700.12  6199.8  704.62  6224.2  707.73  6285.6  712.22  6461.2  718.67
#Mann=3,-1,0
  4411.0    0.06       0  4979.3   0.045       0  5020.7    0.06       0
#XS Ineff=2,0
       0                 5700.00    0.00  708.00
Permanent Ineff=
       F       F
Bank Sta=4979.3,5020.7
XS Rating Curve= 0
Exp/Cntr=0.3,0.1

Type RM Length L Ch R = 1,89685,366,366,366
BEGIN DESCRIPTION:
Dutchman Creek 103.0
END DESCRIPTION:
XS GIS Cut Line= 4
      1544743.48       810108.23      1544125.25       810193.89
      1544024.70       810179.00      1543838.53       810186.44
#Sta/Elev= 30
  4330.4  702.23  4502.7  697.46  4537.6  696.09  4628.1  690.85  4709.5  686.94
  4739.5  686.95  4769.0  685.21  4788.7  683.24  4807.1  680.78  4832.2  676.09
  4891.7  675.87  4907.6  676.77  4959.6  677.05  4964.6  676.96  4978.4  674.76
  4980.1  669.76  5019.9  669.76  5021.6  674.76  5026.9  678.85  5051.2  677.99
  5078.1  678.50  5105.6  683.01  5143.4  695.32  5161.4  700.30  5174.3  703.21
  5191.6  706.02  5206.4  707.51  5218.5  707.13  5230.8  705.88  5242.5  705.83
#Mann=4,-1,0
  4330.4    0.08       0  4628.1    0.14       0  4978.4   0.045       0
  5021.6    0.14       0
Bank Sta=4978.4,5021.6
XS Rating Curve= 0
Exp/Cntr=0.3,0.1

Type RM Length L Ch R = 1,89319,524,524,524
BEGIN DESCRIPTION:
Dutchman Creek 102.0
END DESCRIPTION:
XS GIS Cut Line= 4
      1544806.72       810011.41      1544516.28       810003.96
      1544155.04       809836.38      1543864.59       809828.93
#Sta/Elev= 30
  4484.0  705.50  4659.9  697.69  4720.0  697.75  4754.8  696.49  4819.8  691.06
  4883.1  687.07  4907.0  681.72  4918.8  680.32  4935.6  677.30  4970.4  676.81
  4975.3  674.46  4977.3  669.46  5022.7  669.46  5024.7  674.46  5028.5  676.45
  5051.8  677.50  5102.5  676.29  5125.2  676.70  5138.0  676.24  5157.0  677.11
  5182.2  677.50  5195.9  676.43  5228.0  677.19  5249.0  679.86  5272.7  685.20
  5301.0  690.75  5362.5  699.19  5393.8  702.76  5413.0  704.16  5463.3  705.06
#Mann=4,-1,0
  4484.0    0.08       0  4819.8    0.14       0  4975.3   0.045       0
  5024.7    0.14       0
Bank Sta=4975.3,5024.7
XS Rating Curve= 0
Exp/Cntr=0.3,0.1

Type RM Length L Ch R = 1,88795,286,286,286
BEGIN DESCRIPTION:
Dutchman Creek 101.0
END DESCRIPTION:
XS GIS Cut Line= 5
      1544966.87       809720.93      1544475.31       809538.45
      1544274.21       809490.04      1544028.42       809486.32
      1543682.07       809575.70
#Sta/Elev= 30
  4220.7  707.07  4367.9  696.83  4402.9  688.61  4489.5  689.79  4616.3  688.85
  4759.1  687.49  4769.6  685.93  4780.1  683.19  4795.5  677.80  4811.9  676.22
  4883.8  675.67  4927.0  677.34  4949.8  676.93  4965.5  678.11  4975.3  674.03
  4977.3  669.03  5022.7  669.03  5024.7  674.03  5028.7  676.41  5073.6  677.25
  5147.5  676.74  5177.4  678.22  5225.6  682.58  5292.7  692.45  5323.4  695.90
  5396.3  701.02  5432.8  702.09  5467.1  701.51  5522.3  702.33  5555.4  703.78
#Mann=5,-1,0
  4220.7    0.08       0  4616.3    0.14       0  4975.3   0.045       0
  5024.7    0.14       0  5073.6    0.06       0
Bank Sta=4975.3,5024.7
XS Rating Curve= 0
Exp/Cntr=0.3,0.1

Type RM Length L Ch R = 1,88509,503,503,503
BEGIN DESCRIPTION:
Dutchman Creek 100.0
END DESCRIPTION:
XS GIS Cut Line= 4
      1544728.53       809102.74      1544229.52       809225.63
      1544080.56       809225.63      1543670.92       809091.57
#Sta/Elev= 30
  4394.3  691.77  4448.3  688.25  4494.1  687.23  4528.8  685.81  4549.9  684.31
  4576.5  680.73  4593.4  679.56  4614.0  677.10  4621.1  676.72  4642.9  676.94
  4670.6  675.15  4689.8  674.71  4728.9  675.86  4769.8  675.46  4780.8  674.82
  4810.9  675.72  4867.0  675.93  4877.5  675.60  4891.5  676.37  4908.4  675.98
  4956.9  676.74  4975.3  673.76  4977.3  668.76  5022.7  668.76  5024.7  673.76
  5030.6  676.56  5101.5  680.94  5203.6  683.74  5399.9  691.79  5488.2  696.15
#Mann=3,-1,0
  4394.3    0.14       0  4975.3   0.045       0  5024.7    0.06       0
Bank Sta=4975.3,5024.7
XS Rating Curve= 0
Exp/Cntr=0.3,0.1
