HEC-RAS study Dutchman Creek.prj: Dutchman Creek Limited Detail Study

--- Dutchman Creek.g01 (geometry) --- (continued)

Type RM Length L Ch R = 1,88006,384,384,384
BEGIN DESCRIPTION:
Dutchman Creek 99.0
END DESCRIPTION:
XS GIS Cut Line= 4
      1544810.51       808849.50      1544512.55       808860.67
      1544196.00       808789.91      1543752.88       808745.23
#Sta/Elev= 30
  4649.7  698.56  4687.4  695.06  4800.8  687.72  4883.5  685.07  4901.7  683.47
  4926.2  678.88  4933.9  678.00  4952.5  677.17  4966.0  677.71  4973.1  675.99
  4975.3  673.27  4977.3  668.27  5022.7  668.27  5024.7  673.27  5036.7  677.37
  5038.3  677.41  5124.0  676.10  5192.2  675.92  5229.2  677.02  5238.8  676.77
  5254.3  677.97  5276.5  681.65  5288.0  682.66  5297.6  682.66  5341.2  685.87
  5450.2  691.47  5534.4  694.00  5574.2  696.17  5620.4  697.13  5717.6  702.38
#Mann=4,-1,0
  4649.7    0.14       0  4975.3   0.045       0  5024.7    0.14       0
  5341.2    0.06       0
Bank Sta=4975.3,5024.7
XS Rating Curve= 0
Exp/Cntr=0.3,0.1

Type RM Length L Ch R = 1,87622,524,524,524
BEGIN DESCRIPTION:
Dutchman Creek 98.0
END DESCRIPTION:
XS GIS Cut Line= 5
      1544911.02       808819.70      1544590.76       808659.57
      1544311.45       808573.91      1544196.00       808566.47
      1543913.02       808473.38
#Sta/Elev= 30
  4308.5  705.93  4335.7  704.55  4345.6  703.26  4362.0  702.23  4480.2  691.47
  4547.0  687.03  4605.1  683.32  4637.3  679.91  4659.7  676.12  4695.6  676.40
  4719.3  675.76  4774.5  676.59  4936.4  676.43  4962.4  675.85  4975.2  672.44
  4975.3  672.90  4977.3  667.90  5022.7  667.90  5024.7  672.90  5043.8  677.41
  5056.1  679.16  5094.1  680.50  5103.1  680.32  5133.4  682.16  5178.2  686.50
  5220.8  689.67  5248.6  690.91  5282.1  691.28  5312.3  692.98  5372.3  695.15
#Mann=5,-1,0
  4308.5    0.06       0  4547.0    0.14       0  4975.3   0.045       0
  5024.7    0.14       0  5312.3    0.06       0
Bank Sta=4975.3,5024.7
XS Rating Curve= 0
Exp/Cntr=0.3,0.1

Type RM Length L Ch R = 1,87098,290,290,290
BEGIN DESCRIPTION:
Dutchman Creek 97.0
END DESCRIPTION:
XS GIS Cut Line= 4
      1545026.48       808413.78      1544628.00       808216.40
      1544438.07       808175.44      1543965.13       808208.95
#Sta/Elev= 30
  4497.0  700.12  4533.0  697.04  4586.4  691.51  4743.8  684.03  4811.7  681.94
  4831.0  680.41  4844.3  680.08  4853.8  678.08  4911.0  678.01  4920.0  677.11
  4956.0  676.64  4967.7  675.83  4975.3  672.39  4977.3  667.39  5022.7  667.39
  5024.7  672.39  5031.4  675.27  5037.1  676.24  5084.7  675.39  5164.9  675.51
  5194.9  674.95  5215.4  675.99  5257.1  679.95  5290.1  681.90  5336.8  683.11
  5358.1  684.47  5423.7  687.02  5433.9  688.37  5453.6  688.60  5610.1  694.32
#Mann=5,-1,0
  4497.0    0.06       0  4811.7    0.14       0  4975.3   0.045       0
  5024.7    0.14       0  5084.7    0.06       0
Bank Sta=4975.3,5024.7
XS Rating Curve= 0
Exp/Cntr=0.3,0.1

Type RM Length L Ch R = 1,86808,719,719,719
BEGIN DESCRIPTION:
Dutchman Creek 96.0
END DESCRIPTION:
XS GIS Cut Line= 5
      1545127.89       807712.55      1544901.75       807717.11
      1544470.89       807944.92      1544238.53       808097.16
      1543976.29       808167.99
#Sta/Elev= 30
  4299.3  702.59  4457.9  695.77  4525.5  693.74  4658.3  688.21  4734.4  682.53
  4777.6  680.97  4802.4  679.34  4838.7  678.60  4893.6  675.65  4937.0  675.81
  4946.2  675.21  4960.5  675.11  4975.3  672.29  4977.3  667.29  5022.7  667.29
  5024.7  672.29  5025.4  677.32  5029.6  676.19  5053.8  675.58  5074.7  674.01
  5110.4  673.97  5139.8  676.07  5163.4  679.02  5175.2  679.79  5274.5  680.81
  5317.4  682.91  5336.0  684.58  5346.0  684.74  5392.9  687.86  5562.3  693.24
#Mann=4,-1,0
  4299.3    0.11       0  4946.2    0.06       0  4975.3   0.045       0
  5024.7    0.06       0
Bank Sta=4975.3,5024.7
XS Rating Curve= 0
Exp/Cntr=0.3,0.1

Type RM Length L Ch R = 1,86089,458,458,458
BEGIN DESCRIPTION:
Dutchman Creek 95.0
END DESCRIPTION:
XS GIS Cut Line= 4
      1544892.40       807400.83      1544382.21       807452.96
      1544009.80       807456.69      1543745.35       807486.48
#Sta/Elev= 30
  4154.4  698.20  4259.0  694.66  4325.8  690.62  4389.3  688.01  4478.4  685.67
  4564.8  682.43  4614.7  681.40  4694.6  680.89  4751.0  679.09  4765.9  679.07
  4800.8  676.85  4879.9  674.14  4948.4  675.18  4963.4  672.26  4975.3  672.05
  4977.3  667.05  5022.7  667.05  5024.7  672.05  5025.5  675.04  5027.4  674.74
  5040.3  676.40  5073.0  682.09  5080.4  682.70  5091.8  684.62  5135.2  689.22
  5198.6  693.92  5210.9  694.20  5234.3  696.32  5264.8  696.75  5305.8  698.49
#Mann=3,-1,0
  4154.4    0.11       0  4975.3   0.045       0  5024.7    0.14       0
Bank Sta=4975.3,5024.7
XS Rating Curve= 0
Exp/Cntr=0.3,0.1

Type RM Length L Ch R = 1,85631,547,547,547
BEGIN DESCRIPTION:
Dutchman Creek 94.0
END DESCRIPTION:
XS GIS Cut Line= 4
      1545041.42       807263.04      1544520.00       807214.62
      1544356.14       807181.10      1543812.42       806868.28
#Sta/Elev= 30
  4045.3  702.26  4089.3  701.33  4127.1  699.24  4192.8  697.70  4241.5  694.20
  4258.4  694.30  4456.4  685.60  4524.8  683.69  4661.5  681.02  4684.1  679.08
  4707.1  678.52  4744.7  678.93  4753.4  677.98  4795.7  677.61  4846.5  678.33
  4878.7  677.46  4926.1  674.13  4952.0  674.28  4975.3  671.90  4977.3  666.90
  5022.7  666.90  5024.7  671.90  5032.7  675.79  5049.4  677.58  5078.8  678.36
  5144.7  681.29  5268.4  688.64  5302.8  687.52  5334.2  689.45  5363.5  692.64
#Mann=6,-1,0
  4045.3    0.14       0  4089.3    0.08       0  4524.8    0.14       0
  4975.3   0.045       0  5024.7    0.14       0  5078.8    0.08       0
Bank Sta=4975.3,5024.7
XS Rating Curve= 0
Exp/Cntr=0.3,0.1

Type RM Length L Ch R = 1,85084,830,830,830
BEGIN DESCRIPTION:
Dutchman Creek 93.0
END DESCRIPTION:
XS GIS Cut Line= 3
      1544999.72       806690.94      1544270.58       806578.76
      1543589.52       806698.95
#Sta/Elev= 30
  4427.2  710.35  4510.5  706.33  4569.0  706.06  4598.2  704.36  4666.1  696.15
  4692.7  694.43  4740.4  689.39  4749.4  687.13  4765.7  686.06  4871.6  672.94
  4956.0  675.14  4966.2  674.41  4975.3  671.54  4977.3  666.54  5022.7  666.54
  5024.7  671.54  5028.2  673.91  5035.7  675.26  5097.2  673.84  5184.9  676.80
  5228.6  682.21  5246.3  683.35  5471.2  687.76  5537.4  691.08  5560.8  691.10
  5684.5  695.37  5710.3  698.06  5740.5  697.05  5756.5  698.68  5856.5  700.46
#Mann=3,-1,0
  4427.2    0.14       0  4975.3   0.045       0  5024.7    0.08       0
Bank Sta=4975.3,5024.7
XS Rating Curve= 0
Exp/Cntr=0.3,0.1

Type RM Length L Ch R = 1,84254,448,448,448
BEGIN DESCRIPTION:
Dutchman Creek 92.0
END DESCRIPTION:
XS GIS Cut Line= 5
      1544870.10       805911.19      1544564.69       805903.74
      1544419.45       805955.88      1543976.28       806056.43
      1543778.87       806048.98
#Sta/Elev= 30
  4613.1  689.37  4646.5  690.33  4695.5  689.45  4706.6  688.21  4716.4  685.37
  4733.3  682.99  4750.6  674.71  4777.8  675.81  4810.7  675.30  4827.4  676.47
  4870.7  674.19  4905.2  675.65  4943.8  675.64  4945.2  675.24  4947.6  670.24
  4975.2  670.80  4977.2  665.80  5022.8  665.80  5024.8  670.80  5029.3  675.07
  5066.5  676.47  5107.5  674.29  5160.6  675.03  5200.6  677.63  5226.1  678.17
  5434.5  678.56  5517.7  684.05  5617.8  698.29  5673.4  705.94  5724.9  708.77
#Mann=4,-1,0
  4613.1    0.14       0  4975.2   0.045       0  5024.8    0.14       0
  5617.8    0.14       0
Bank Sta=4975.2,5024.8
XS Rating Curve= 0
Exp/Cntr=0.3,0.1

Type RM Length L Ch R = 1,83806,304,304,304
BEGIN DESCRIPTION:
Dutchman Creek 91.0
END DESCRIPTION:
XS GIS Cut Line= 5
      1545352.29       806114.03      1544844.00       805747.33
      1544549.79       805643.05      1544017.25       805423.33
      1543864.56       805237.12
#Sta/Elev= 30
  3801.7  706.36  3831.4  704.05  3855.7  700.79  3932.8  694.96  4083.5  686.69
  4132.7  685.67  4232.3  686.78  4355.4  687.16  4585.2  683.28  4647.5  679.23
  4698.9  673.62  4762.4  673.94  4829.7  676.65  4882.7  674.85  4931.1  674.97
  4947.5  670.16  4952.3  670.13  4975.2  670.40  4977.2  665.40  5022.8  665.40
  5024.8  670.40  5033.4  675.27  5050.7  676.72  5088.4  675.04  5123.0  675.13
  5187.5  675.91  5271.4  679.59  5300.3  678.98  5327.1  684.23  5557.5  713.45
#Mann=5,-1,0
  3801.7    0.06       0  4232.3    0.14       0  4952.3    0.08       0
  4975.2   0.045       0  5024.8    0.08       0
#XS Ineff=2,0
    0.00 4581.80  704.05               0
Permanent Ineff=
       F       F
Bank Sta=4975.2,5024.8
XS Rating Curve= 0
Exp/Cntr=0.5,0.3

Type RM Length L Ch R = 1,83502,312,312,312
BEGIN DESCRIPTION:
I-40 (DC) us
END DESCRIPTION:
XS GIS Cut Line= 5
      1545662.33       806095.75      1545186.96       805861.67
      1544434.26       805267.44      1544272.20       805065.76
      1543912.08       804716.44
#Sta/Elev= 30
  3613.9  689.88  3663.6  688.72  3729.1  694.71  3817.5  697.71  3976.6  693.32
  4053.6  688.77  4281.9  682.96  4406.1  683.86  4640.7  677.36  4707.4  673.75
  4761.8  676.01  4898.1  673.77  4969.8  676.07  4976.0  672.23  4986.5  665.13
  5013.5  665.13  5024.0  672.23  5027.8  673.84  5119.5  674.71  5146.7  678.84
  5198.1  679.06  5275.0  682.84  5364.3  684.07  5374.4  688.21  5440.9  684.24
  5471.1  689.53  5564.5  695.35  5583.3  695.60  5710.7  688.53  5863.2  690.46
#Mann=6,-1,0
  3613.9    0.14       0  3976.6    0.06       0  4281.9    0.14       0
  4976.0   0.045       0  5024.0    0.14       0  5198.1    0.06       0
#XS Ineff=2,0
    0.00 4832.50  689.80 5167.50    0.00  690.05
Permanent Ineff=
       F       F
Bank Sta=4976,5024
XS Rating Curve= 0
Exp/Cntr=0.5,0.3

Type RM Length L Ch R =3,83361,,,
BEGIN DESCRIPTION:
I-40 (DC) tor
Structure ID: LDS_DC_08
Approximate Survey Structure
END DESCRIPTION:
Bridge Culvert--1,0,-1,-1,0
Deck Dist Width WeirC Skew NumUp NumDn MinLoCord MaxHiCord MaxSubmerge Is_Ogee
76,130,3,,11,11,,,0.95,0,1,1,,,
  3568.3  3877.1  4258.0  4908.5  4908.5  5091.5  5091.5  5479.1  5698.7  5856.9
  5951.3
  690.76  689.84  690.15  690.13  690.13  690.13  690.13  689.98  690.15  691.16
  691.76
  645.13  645.13  645.13  645.13  686.53  686.53  645.13  645.13  645.13  645.13
  645.13
  3568.3  3877.1  4258.0  4908.5  4908.5  5091.5  5091.5  5479.1  5698.7  5856.9
  5951.3
  690.76  689.84  690.15  690.13  690.13  690.13  690.13  689.98  690.15  691.16
  691.76
  645.13  645.13  645.13  645.13  686.53  686.53  645.13  645.13  645.13  645.13
  645.13
Pier Skew, UpSta & Num, DnSta & Num=,4954.3,2,4954.3,2,0,0,0,0,0
     2.8     2.8
  675.11  686.53
     2.8     2.8
  671.99  686.53
Pier Skew, UpSta & Num, DnSta & Num=,5045.8,2,5045.8,2,0,0,0,0,0
     2.8     2.8
  673.34  686.53
     2.8     2.8
  675.45  686.53
Abutment Skew #Up #Dn=,2,2
  4908.5  4932.5
  686.53  674.76
  4908.5  4932.5
  686.53  671.58
Abutment Skew #Up #Dn=,2,2
  5067.5  5091.5
  673.15  686.53
  5067.5  5091.5
  674.76  686.53
BR Coef=1,1,0,1.25,0,,,0.8,0,2,0,
WSPro=,,,, 1 ,,,, 0 ,,,, 0 ,,,,-1 ,-1 ,-1 , 0 , 0 , 0 , 0 , 0
BC Design=,,0,,0,,,,,,

Type RM Length L Ch R = 1,83190,908,908,908
BEGIN DESCRIPTION:
I-40 (DC) ds
END DESCRIPTION:
XS GIS Cut Line= 4
      1545640.73       806023.73      1545532.69       805724.81
      1544322.62       804792.05      1543976.92       804644.41
#Sta/Elev= 30
  3623.5  690.62  3717.7  688.26  3770.0  690.47  3867.9  689.11  3927.3  679.61
  3984.3  678.20  4017.6  675.21  4064.1  676.98  4097.6  672.97  4124.1  676.61
  4151.2  677.23  4608.0  676.85  4679.2  674.99  4747.6  677.55  4773.2  673.87
  4828.7  672.12  4957.5  672.16  4969.2  671.95  4974.8  669.67  4976.0  671.98
  4986.5  664.88  5013.5  664.88  5024.0  671.98  5043.7  675.52  5089.1  673.34
  5164.8  675.33  5217.8  672.68  5484.4  676.43  5631.0  686.76  5845.1  690.78
#Mann=3,-1,0
  3623.5    0.14       0  4976.0   0.045       0  5024.0    0.06       0
#XS Ineff=2,0
    0.00 4802.50  689.78 5197.50    0.00  690.03
Permanent Ineff=
       F       F
Bank Sta=4976,5024
XS Rating Curve= 0
Exp/Cntr=0.5,0.3

Type RM Length L Ch R = 1,82282,709,709,709
BEGIN DESCRIPTION:
Dutchman Creek 90.0
END DESCRIPTION:
XS GIS Cut Line= 4
      1545231.32       804268.86      1544989.24       804291.21
      1544680.14       804402.93      1543972.54       804596.59
#Sta/Elev= 30
  4682.0  712.07  4774.7  706.22  4804.9  702.02  4831.5  697.22  4863.9  688.65
  4891.7  682.91  4912.7  678.47  4966.2  675.73  4975.2  669.79  4977.2  664.79
  5022.8  664.79  5024.8  669.79  5032.2  673.99  5049.9  674.80  5073.5  673.96
  5145.6  674.02  5191.4  672.11  5256.3  673.61  5329.6  672.49  5351.8  673.04
  5405.7  671.33  5423.8  673.49  5497.4  676.23  5581.9  674.78  5656.5  675.59
  5770.3  680.23  5798.6  679.77  5849.3  681.40  5960.4  687.53  5987.4  689.82
#Mann=4,-1,0
  4682.0     0.1       0  4891.7    0.06       0  4975.2   0.045       0
  5024.8    0.06       0
#XS Ineff=2,0
       0                 5491.10    0.00  693.63
Permanent Ineff=
       F       F
Bank Sta=4975.2,5024.8
XS Rating Curve= 0
Exp/Cntr=0.3,0.1

Type RM Length L Ch R = 1,81573,543,543,543
BEGIN DESCRIPTION:
Dutchman Creek 89.0
END DESCRIPTION:
XS GIS Cut Line= 5
      1545261.14       803877.83      1545071.17       803915.08
      1544520.00       803889.01      1543972.56       803929.97
      1543760.29       804172.04
#Sta/Elev= 30
  4319.3  707.72  4352.5  704.02  4379.1  702.70  4425.9  694.78  4448.0  689.06
  4476.3  677.95  4490.1  674.13  4497.9  673.33  4594.6  671.87  4662.8  672.60
  4706.1  672.23  4714.9  671.47  4798.7  673.23  4877.2  672.31  4931.5  673.65
  4973.9  672.62  4975.2  669.32  4977.2  664.32  5022.8  664.32  5024.8  669.32
  5029.5  674.44  5146.8  673.03  5195.4  673.91  5418.0  671.95  5552.1  673.16
  5622.1  676.85  5653.7  677.07  5753.3  681.09  5893.4  689.26  5935.6  692.90
#Mann=4,-1,0
  4319.3     0.1       0  4594.6    0.06       0  4975.2   0.045       0
  5024.8    0.06       0
#XS Ineff=2,0
       0                 5366.90    0.00  689.13
Permanent Ineff=
       F       F
Bank Sta=4975.2,5024.8
XS Rating Curve= 0
Exp/Cntr=0.3,0.1

Type RM Length L Ch R = 1,81030,545,545,545
BEGIN DESCRIPTION:
Dutchman Creek 88.0
END DESCRIPTION:
XS GIS Cut Line= 4
      1545253.05       803726.81      1544996.68       803620.87
      1544810.48       803397.43      1544743.46       803174.02
#Sta/Elev= 30
  4471.0  707.37  4558.0  699.41  4603.8  692.84  4625.0  691.19  4668.8  685.96
  4680.3  685.65  4739.7  675.48  4754.9  673.84  4767.8  673.63  4782.5  672.31
  4860.2  671.61  4883.1  672.27  4924.5  670.95  4955.4  671.95  4963.5  671.35
  4974.9  668.73  4976.9  663.73  5023.1  663.73  5025.1  668.73  5028.8  670.25
  5070.9  670.38  5106.7  671.92  5113.5  673.73  5132.0  680.95  5160.1  695.61
  5179.2  701.61  5205.4  707.33  5213.4  711.08  5232.1  717.35  5272.5  718.98
#Mann=4,-1,0
  4471.0     0.1       0  4739.7    0.14       0  4974.9   0.045       0
  5025.1    0.14       0
Bank Sta=4974.9,5025.1
XS Rating Curve= 0
Exp/Cntr=0.5,0.3

Type RM Length L Ch R = 1,80485,133,133,133
BEGIN DESCRIPTION:
US 158 (DC) us
END DESCRIPTION:
XS GIS Cut Line= 5
      1545654.17       803592.49      1545406.51       803290.72
      1545156.75       802984.76      1545117.20       802872.37
      1545002.71       802693.34
#Sta/Elev= 30
  4337.7  706.58  4387.7  704.81  4497.1  698.40  4557.0  691.48  4566.9  692.55
  4599.9  688.96  4664.9  683.86  4727.0  679.66  4760.5  679.17  4818.8  674.81
  4919.6  671.54  4928.7  668.40  4934.4  670.88  4970.9  670.65  4975.0  669.84
  4980.5  663.14  5019.5  663.14  5025.0  669.84  5026.6  671.96  5033.9  674.07
  5063.0  680.36  5108.5  681.35  5123.0  684.67  5134.7  685.45  5180.6  685.73
  5211.8  690.42  5324.0  687.22  5335.4  688.72  5364.6  690.05  5454.7  692.45
#Mann=4,-1,0
  4337.7     0.1       0  4664.9    0.14       0  4975.0   0.045       0
  5025.0    0.14       0
#XS Ineff=2,0
    0.00 4878.50  682.94 5121.50    0.00  683.21
Permanent Ineff=
       F       F
Bank Sta=4975,5025
XS Rating Curve= 0
Exp/Cntr=0.5,0.3

Type RM Length L Ch R =3,80416,,,
BEGIN DESCRIPTION:
US 158 (DC) tor
Structure ID: LDS_DC_06
Approximate Survey Structure
END DESCRIPTION:
Bridge Culvert--1,0,-1,-1,0
Deck Dist Width WeirC Skew NumUp NumDn MinLoCord MaxHiCord MaxSubmerge Is_Ogee
53.5,31,3,,18,18,,,0.95,0,1,1,,,
  4333.4  4433.5  4580.9  4676.0  4754.2  4820.0  4867.0  4920.5  4932.0  4932.0
  5068.0  5068.0  5078.2  5119.3  5169.8  5218.5  5386.7  5493.2
  707.62  703.19  694.82  689.68  686.09  683.97  683.14  682.84  682.84  682.84
  682.84  682.84  682.84  683.21  684.01  685.04  689.80  693.98
  643.14  643.14  643.14  643.14  643.14  643.14  643.14  643.14  643.14  679.34
  679.34  643.14  643.14  643.14  643.14  643.14  643.14  643.14
  4333.4  4433.5  4580.9  4676.0  4754.2  4820.0  4867.0  4920.5  4932.0  4932.0
  5068.0  5068.0  5078.2  5119.3  5169.8  5218.5  5386.7  5493.2
  707.62  703.19  694.82  689.68  686.09  683.97  683.14  682.84  682.84  682.84
  682.84  682.84  682.84  683.21  684.01  685.04  689.80  693.98
  643.14  643.14  643.14  643.14  643.14  643.14  643.14  643.14  643.14  679.34
  679.34  643.14  643.14  643.14  643.14  643.14  643.14  643.14
Pier Skew, UpSta & Num, DnSta & Num=,4966,2,4966,2,0,0,0,0,0
       3       3
  670.69  679.34
       3       3
  671.18  679.34
Pier Skew, UpSta & Num, DnSta & Num=,5034,2,5034,2,0,0,0,0,0
       3       3
  674.09  679.34
       3       3
  671.74  679.34
Abutment Skew #Up #Dn=,2,2
  4932.0  4935.0
  679.34  670.84
  4932.0  4935.0
  679.34  672.35
Abutment Skew #Up #Dn=,2,2
  5065.0  5068.0
  680.42  679.34
  5065.0  5068.0
  674.00  679.34
BR Coef=1,1,0,1.25,0,,,0.8,0,2,0,
WSPro=,,,, 1 ,,,, 0 ,,,, 0 ,,,,-1 ,-1 ,-1 , 0 , 0 , 0 , 0 , 0
BC Design=,,0,,0,,,,,,

Type RM Length L Ch R = 1,80352,118,118,118
BEGIN DESCRIPTION:
US 158 (DC) ds
END DESCRIPTION:
XS GIS Cut Line= 5
      1545714.56       803505.11      1545500.17       803232.44
      1545439.81       803130.46      1545196.29       802822.42
      1545017.31       802678.82
#Sta/Elev= 30
  4392.6  711.67  4415.1  710.77  4438.8  711.78  4485.5  707.86  4490.4  709.43
  4509.4  708.85  4538.6  703.19  4552.3  707.35  4560.2  704.74  4585.7  703.90
  4598.2  699.41  4624.4  697.40  4649.1  698.82  4657.6  695.68  4679.8  695.14
  4713.3  692.42  4724.6  693.18  4767.0  684.77  4789.1  683.25  4813.1  678.94
  4858.5  675.69  4970.0  671.14  4975.0  669.59  4980.5  662.89  5019.5  662.89
  5025.0  669.59  5054.7  674.02  5257.1  677.43  5289.0  682.99  5480.1  692.71
#Mann=4,-1,0
  4392.6     0.1       0  4679.8    0.14       0  4975.0   0.045       0
  5025.0    0.14       0
#XS Ineff=2,0
    0.00 4883.50  682.99 5116.50    0.00  683.19
Permanent Ineff=
       F       F
Bank Sta=4975,5025
XS Rating Curve= 0
Exp/Cntr=0.5,0.3

Type RM Length L Ch R = 1,80234,723,723,723
BEGIN DESCRIPTION:
Dutchman Creek 87.0
END DESCRIPTION:
XS GIS Cut Line= 4
      1545723.38       803257.77      1545516.05       803034.18
      1545227.43       802676.45      1545028.22       802550.42
#Sta/Elev= 30
  4579.1  712.73  4641.6  710.84  4689.9  705.23  4705.4  704.29  4738.3  698.26
  4761.1  695.91  4798.8  689.36  4813.4  685.80  4868.4  681.99  4879.3  679.79
  4896.2  672.76  4925.3  670.17  4934.4  668.25  4940.2  670.32  4947.9  671.42
  4974.9  668.84  4977.3  662.84  5022.7  662.84  5025.1  668.84  5053.7  680.49
  5065.1  681.52  5197.2  681.95  5219.8  681.19  5229.1  681.83  5250.9  681.30
  5389.2  682.62  5462.3  685.81  5533.7  691.39  5566.4  694.84  5579.4  695.19
#Mann=4,-1,0
  4579.1    0.06       0  4689.9    0.14       0  4974.9   0.045       0
  5025.1    0.14       0
Bank Sta=4974.9,5025.1
XS Rating Curve= 0
Exp/Cntr=0.3,0.1

Type RM Length L Ch R = 1,79511,673,673,673
BEGIN DESCRIPTION:
Dutchman Creek 86.0
END DESCRIPTION:
XS GIS Cut Line= 3
      1545903.44       803069.62      1545978.75       802768.38
      1545403.69       801953.70
#Sta/Elev= 30
  4266.2  692.24  4318.7  691.34  4328.1  690.57  4345.9  686.46  4361.0  684.61
  4438.2  684.98  4504.8  684.09  4576.7  680.30  4613.9  677.26  4791.3  669.84
  4912.8  670.60  4946.6  671.97  4960.2  671.62  4969.3  668.76  4974.9  668.43
  4977.3  662.43  5022.7  662.43  5025.1  668.43  5030.5  672.74  5109.0  673.01
  5249.1  671.53  5276.1  673.20  5300.9  673.17  5322.7  675.06  5355.5  677.97
  5384.3  679.28  5424.5  686.86  5477.9  694.62  5553.1  701.66  5573.9  705.47
#Mann=4,-1,0
  4266.2    0.06       0  4974.9   0.045       0  5025.1    0.06       0
  5322.7    0.14       0
#XS Ineff=2,0
       0                 5226.70    0.00  690.04
Permanent Ineff=
       F       F
Bank Sta=4974.9,5025.1
XS Rating Curve= 0
Exp/Cntr=0.3,0.1

Type RM Length L Ch R = 1,78838,447,447,447
BEGIN DESCRIPTION:
Dutchman Creek 85.0
END DESCRIPTION:
XS GIS Cut Line= 4
      1546542.18       803192.60      1546531.01       802909.57
      1546333.63       802283.92      1546225.63       801669.44
#Sta/Elev= 30
  4103.6  688.68  4173.3  682.21  4301.0  675.35  4382.5  673.63  4411.7  670.69
  4437.7  672.12  4738.7  671.40  4762.8  668.50  4786.8  671.47  4883.0  668.80
  4968.2  671.05  4974.9  667.69  4977.3  661.69  5022.7  661.69  5025.1  667.69
  5035.1  667.42  5054.9  669.89  5084.4  669.81  5085.7  668.93  5086.1  667.39
  5162.4  670.82  5192.0  670.00  5233.7  671.42  5396.9  672.63  5473.9  674.86
  5486.3  676.82  5519.1  686.48  5562.5  695.83  5612.5  702.86  5666.8  706.61
#Mann=4,-1,0
  4103.6    0.06       0  4974.9   0.045       0  5025.1    0.06       0
  5396.9    0.14       0
#XS Ineff=2,0
    0.00 4605.60  693.48 5220.10    0.00  693.48
Permanent Ineff=
       F       F
Bank Sta=4974.9,5025.1
XS Rating Curve= 0
Exp/Cntr=0.3,0.1

Type RM Length L Ch R = 1,78391,403,403,403
BEGIN DESCRIPTION:
Dutchman Creek 84.0
END DESCRIPTION:
XS GIS Cut Line= 4
      1546986.76       802568.49      1546843.83       802466.41
      1546743.28       802201.99      1546810.32       801956.20
#Sta/Elev= 30
  4679.6  689.23  4704.2  688.03  4727.8  684.47  4763.0  681.61  4774.7  678.07
  4808.6  674.94  4834.5  674.22  4858.7  669.55  4871.3  670.47  4878.1  668.85
  4883.6  668.67  4898.0  670.09  4928.9  671.31  4960.3  669.88  4974.9  667.27
  4977.3  661.27  5022.7  661.27  5025.1  667.27  5031.2  670.35  5039.0  671.72
  5066.0  671.20  5096.1  673.96  5104.3  675.69  5109.6  678.36  5132.9  683.90
  5156.0  692.44  5172.0  693.85  5230.9  695.02  5322.2  700.66  5392.9  702.79
#Mann=3,-1,0
  4679.6    0.14       0  4974.9   0.045       0  5025.1    0.14       0
Bank Sta=4974.9,5025.1
XS Rating Curve= 0
Exp/Cntr=0.3,0.1

Type RM Length L Ch R = 1,77988,527,527,527
BEGIN DESCRIPTION:
Dutchman Creek 83.0
END DESCRIPTION:
XS GIS Cut Line= 3
      1547354.22       802552.45      1547110.28       802078.58
      1547152.35       801820.56
#Sta/Elev= 30
  4558.7  706.46  4720.8  693.50  4740.2  690.50  4764.6  688.18  4786.2  684.32
  4832.0  679.52  4844.7  676.17  4867.7  671.53  4891.6  670.11  4914.9  670.78
  4935.5  669.68  4943.9  670.39  4955.0  670.08  4964.8  669.19  4972.4  669.31
  4974.9  667.07  4977.3  661.07  5022.7  661.07  5025.1  667.07  5041.0  671.36
  5060.7  674.70  5075.9  676.58  5093.5  681.43  5133.3  687.06  5159.5  689.93
  5185.3  691.11  5216.6  695.73  5259.8  700.86  5328.7  707.52  5353.1  709.35
#Mann=3,-1,0
  4558.7    0.14       0  4974.9   0.045       0  5025.1    0.14       0
Bank Sta=4974.9,5025.1
XS Rating Curve= 0
Exp/Cntr=0.3,0.1

Type RM Length L Ch R = 1,77461,413,413,413
BEGIN DESCRIPTION:
Dutchman Creek 82.0
END DESCRIPTION:
XS GIS Cut Line= 4
      1547819.51       802142.39      1547715.27       802094.00
      1547566.31       801859.38      1547406.41       801682.20
#Sta/Elev= 30
  4767.0  686.89  4817.6  684.69  4841.6  684.74  4872.0  681.69  4904.8  678.85
  4916.5  675.60  4935.1  672.67  4952.1  668.78  4965.3  669.17  4974.9  666.78
  4977.3  660.78  5022.7  660.78  5025.1  666.78  5039.9  669.97  5076.5  672.02
  5102.4  671.24  5114.1  669.83  5127.3  669.74  5148.9  670.43  5163.7  671.57
  5176.6  674.09  5187.2  676.79  5199.3  679.02  5215.9  683.44  5271.2  695.96
  5295.9  700.44  5304.4  702.75  5329.0  706.51  5353.5  709.71  5398.5  711.52
#Mann=4,-1,0
  4767.0    0.08       0  4872.0    0.14       0  4974.9   0.045       0
  5025.1    0.14       0
Bank Sta=4974.9,5025.1
XS Rating Curve= 0
Exp/Cntr=0.3,0.1

Type RM Length L Ch R = 1,77048,657,657,657
BEGIN DESCRIPTION:
Dutchman Creek 81.0
END DESCRIPTION:
XS GIS Cut Line= 4
      1548106.30       802008.33      1548076.51       801848.21
      1547774.86       801557.73      1547428.49       801464.62
#Sta/Elev= 30
  4696.8  690.15  4742.4  687.10  4793.9  682.45  4810.5  679.30  4842.9  676.17
  4884.1  670.39  4907.7  669.42  4928.7  671.72  4941.9  669.21  4952.9  670.16
  4965.6  668.75  4974.9  666.55  4977.3  660.55  5022.7  660.55  5025.1  666.55
  5046.2  671.84  5088.3  670.18  5109.8  671.12  5166.6  670.88  5181.9  669.67
  5240.0  670.65  5369.7  678.49  5396.1  682.45  5426.9  689.73  5448.9  692.97
  5464.6  699.89  5476.4  703.38  5528.9  713.55  5569.2  719.54  5637.1  726.32
#Mann=4,-1,0
  4696.8    0.09       0  4742.4    0.08       0  4974.9   0.045       0
  5025.1    0.14       0
Bank Sta=4974.9,5025.1
XS Rating Curve= 0
Exp/Cntr=0.3,0.1

Type RM Length L Ch R = 1,76391,1097,1097,1097
BEGIN DESCRIPTION:
Dutchman Creek 80.0
END DESCRIPTION:
XS GIS Cut Line= 4
      1549245.49       801956.29      1548839.38       801524.80
      1547910.41       801197.24      1547660.17       801158.51
#Sta/Elev= 30
  4019.8  699.16  4150.0  692.33  4186.2  688.68  4257.9  686.84  4409.7  687.05
  4440.0  690.01  4510.3  688.62  4660.0  679.39  4705.7  678.27  4789.5  669.21
  4824.9  667.77  4961.1  670.72  4969.0  669.64  4974.8  666.14  4977.2  660.14
  5022.8  660.14  5025.2  666.14  5033.4  665.82  5043.4  665.44  5052.1  669.28
  5083.8  667.32  5209.0  668.29  5236.7  669.99  5322.7  668.25  5406.9  671.83
  5524.3  671.17  5567.5  672.62  5657.1  677.56  5802.0  695.38  5850.6  695.64
#Mann=4,-1,0
  4019.8    0.09       0  4974.8   0.045       0  5025.2    0.09       0
  5033.4    0.14       0
Bank Sta=4974.8,5025.2
XS Rating Curve= 0
Exp/Cntr=0.3,0.1

Type RM Length L Ch R = 1,75294,923,923,923
BEGIN DESCRIPTION:
Dutchman Creek 79.0
END DESCRIPTION:
XS GIS Cut Line= 4
      1550387.75       800264.12      1548340.19       800331.81
      1547552.22       800358.16      1547138.75       800424.87
#Sta/Elev= 30
  2956.8  712.26  3063.6  706.49  3236.1  701.01  3345.3  691.46  3421.8  690.13
  3486.2  682.11  3534.6  673.48  3654.8  666.82  4029.1  669.47  4239.5  668.86
  4351.0  666.44  4475.5  668.63  4485.8  666.96  4657.7  666.68  4959.7  669.16
  4964.0  665.43  4974.8  665.43  4977.2  659.43  5022.8  659.43  5025.2  665.43
  5038.9  669.44  5057.5  669.11  5196.5  668.73  5319.8  665.97  5361.0  667.51
  5386.7  665.51  5854.8  676.43  6023.1  687.95  6115.4  697.15  6212.7  714.90
#Mann=4,-1,0
  2956.8    0.06       0  4974.8   0.045       0  5025.2    0.06       0
  5057.5     0.1       0
#XS Ineff=2,0
    0.00 4035.40  693.85 5699.80    0.00  693.85
Permanent Ineff=
       F       F
Bank Sta=4974.8,5025.2
XS Rating Curve= 0
Exp/Cntr=0.3,0.1

Type RM Length L Ch R = 1,74371,1247,1247,1247
BEGIN DESCRIPTION:
Dutchman Creek 78.0
END DESCRIPTION:
XS GIS Cut Line= 5
      1549663.55       799322.71      1549289.42       799614.71
      1548655.28       799623.84      1548459.11       799546.28
      1547460.21       799617.70
#Sta/Elev= 30
  3781.7  706.33  3860.1  701.04  3895.7  698.99  3916.4  695.28  3973.4  680.46
  4045.8  667.65  4077.2  665.14  4088.7  668.46  4150.1  671.02  4209.4  679.44
  4243.0  681.08  4312.6  677.49  4323.2  675.44  4342.7  667.65  4367.5  665.75
  4667.2  667.09  4816.9  667.16  4854.2  665.53  4938.3  668.44  4944.7  665.42
  4974.8  664.58  4977.2  658.58  5022.8  658.58  5025.2  664.58  5050.4  665.42
  5058.2  671.42  5262.9  672.00  5518.3  684.05  5802.9  683.11  6102.9  695.79
#Mann=8,-1,0
  3781.7    0.06       0  3860.1    0.14       0  4088.7    0.06       0
  4667.2    0.14       0  4974.8   0.045       0  5025.2    0.14       0
  5262.9    0.14       0  5518.3    0.06       0
#XS Ineff=2,0
    0.00 4255.50  688.37 5526.20    0.00  688.37
Permanent Ineff=
       F       F
Bank Sta=4974.8,5025.2
XS Rating Curve= 0
Exp/Cntr=0.3,0.1

Type RM Length L Ch R = 1,73124,944,944,944
BEGIN DESCRIPTION:
Dutchman Creek 77.0
END DESCRIPTION:
XS GIS Cut Line= 6
      1549451.30       799076.59      1549321.12       798976.79
      1549203.94       798968.11      1548787.27       799167.76
      1547806.37       799358.73      1547415.73       799597.46
#Sta/Elev= 30
  4659.5  690.95  4781.0  689.08  4838.9  686.08  4931.5  670.80  4969.0  667.95
  4973.5  666.48  4974.8  663.42  4977.2  657.42  5022.8  657.42  5025.2  663.42
  5028.5  665.35  5034.6  666.42  5053.2  667.86  5170.5  668.29  5301.0  666.45
  5353.5  667.17  5578.8  667.75  5698.1  667.07  5715.9  668.13  5820.0  666.42
  5983.8  666.38  6052.6  674.66  6081.4  680.21  6113.1  681.94  6185.2  681.35
  6274.1  682.38  6427.4  681.03  6529.4  682.11  6690.6  686.38  6860.2  696.74
#Mann=6,-1,0
  4659.5    0.14       0  4974.8   0.045       0  5025.2    0.14       0
  5353.5    0.06       0  5578.8    0.14       0  6081.4    0.06       0
Bank Sta=4974.8,5025.2
XS Rating Curve= 0
Exp/Cntr=0.3,0.1

Type RM Length L Ch R = 1,72180,928,928,928
BEGIN DESCRIPTION:
Dutchman Creek 76.0
END DESCRIPTION:
XS GIS Cut Line= 4
      1549389.37       798966.24      1549230.76       798741.58
      1549143.17       798438.60      1548379.26       797796.22
#Sta/Elev= 30
  4545.0  691.42  4563.2  692.29  4660.8  687.44  4698.7  683.25  4757.8  677.93
  4807.2  671.48  4861.6  667.40  4907.9  666.06  4953.8  665.97  4971.4  664.55
  4975.0  656.55  5025.0  656.55  5028.6  664.55  5078.9  666.56  5161.8  665.26
  5182.7  666.15  5287.9  665.79  5399.3  667.10  5443.5  666.65  5580.6  666.05
  5706.1  666.66  5725.7  666.04  5838.8  666.40  5876.6  667.31  5909.3  672.84
  5940.4  681.17  5988.3  692.47  6011.7  696.41  6037.3  698.19  6133.5  701.36
#Mann=4,-1,0
  4545.0    0.14       0  4971.4   0.045       0  5028.6    0.14       0
  5443.5    0.14       0
Bank Sta=4971.4,5028.6
XS Rating Curve= 0
Exp/Cntr=0.3,0.1

Type RM Length L Ch R = 1,71252,1162,1162,1162
BEGIN DESCRIPTION:
Dutchman Creek 75.0
END DESCRIPTION:
XS GIS Cut Line= 4
      1550132.76       798933.39      1549746.47       798677.31
      1549551.16       798325.75      1549650.98       797787.56
#Sta/Elev= 30
  3778.8  703.31  3858.9  698.26  3921.3  695.31  3976.5  694.02  4000.5  694.74
  4019.5  693.75  4090.9  685.69  4126.4  680.49  4151.1  674.63  4183.6  669.28
  4221.9  665.67  4262.5  664.63  4281.3  663.30  4401.5  664.92  4442.6  666.21
  4606.5  664.47  4797.1  665.01  4908.8  666.29  4936.0  665.99  4971.4  663.54
  4975.0  655.54  5025.0  655.54  5028.6  663.54  5054.9  668.41  5078.0  679.31
  5097.3  686.94  5105.0  688.71  5120.5  696.33  5143.1  704.62  5191.8  720.18
#Mann=3,-1,0
  3778.8    0.14       0  4971.4   0.045       0  5028.6    0.14       0
Bank Sta=4971.4,5028.6
XS Rating Curve= 0
Exp/Cntr=0.3,0.1

Type RM Length L Ch R = 1,70090,796,796,796
BEGIN DESCRIPTION:
Dutchman Creek 74.0
END DESCRIPTION:
XS GIS Cut Line= 4
      1550321.76       798826.75      1550162.68       798449.66
      1549897.56       797866.40      1549697.22       797630.70
#Sta/Elev= 30
  4705.4  719.36  4805.1  714.45  4914.1  695.56  4927.7  692.27  4942.9  685.87
  4959.7  673.82  4966.7  670.06  4971.4  662.65  4975.0  654.65  5025.0  654.65
  5028.6  662.65  5044.8  662.54  5049.7  663.93  5143.8  663.12  5173.1  664.05
  5197.8  662.87  5226.9  664.63  5290.2  663.23  5325.3  664.54  5414.8  664.14
  5579.5  666.17  5733.7  665.94  5772.1  666.11  5785.9  667.92  5803.0  671.85
  5846.7  687.43  5918.7  717.11  5965.6  731.98  6002.7  737.25  6064.7  743.56
#Mann=4,-1,0
  4705.4    0.14       0  4971.4   0.045       0  5028.6    0.14       0
  5733.7     0.1       0
Bank Sta=4971.4,5028.6
XS Rating Curve= 0
Exp/Cntr=0.3,0.1

Type RM Length L Ch R = 1,69294,607,607,607
BEGIN DESCRIPTION:
Dutchman Creek 73.0
END DESCRIPTION:
XS GIS Cut Line= 5
      1551456.57       798437.74      1551161.40       798277.14
      1550579.80       798073.14      1550341.09       797860.47
      1550054.66       797482.90
#Sta/Elev= 30
  4151.7  714.13  4205.2  710.20  4260.5  704.21  4314.3  701.77  4321.4  699.98
  4364.8  696.91  4413.3  689.70  4457.3  679.38  4515.8  669.44  4548.6  668.55
  4828.3  664.29  4929.2  664.65  4971.4  662.16  4975.0  654.16  5025.0  654.16
  5028.6  662.16  5043.2  664.26  5078.2  664.72  5168.2  662.91  5230.8  663.59
  5344.0  667.51  5416.5  665.26  5583.6  665.33  5618.2  669.62  5685.6  692.33
  5759.1  711.54  5806.9  719.94  5841.4  724.33  5867.4  726.40  5897.7  726.72
#Mann=5,-1,0
  4151.7    0.14       0  4548.6    0.08       0  4971.4   0.045       0
  5028.6    0.08       0  5618.2     0.1       0
Bank Sta=4971.4,5028.6
XS Rating Curve= 0
Exp/Cntr=0.3,0.1

Type RM Length L Ch R = 1,68687,989,989,989
BEGIN DESCRIPTION:
Dutchman Creek 72.0
END DESCRIPTION:
XS GIS Cut Line= 4
      1551582.52       798013.67      1551352.77       797766.24
      1550410.12       797371.51      1550080.22       797442.20
#Sta/Elev= 30
  4118.0  716.11  4187.2  710.47  4207.9  707.00  4311.3  695.42  4367.6  687.66
  4399.9  682.12  4438.9  671.72  4480.8  663.91  4512.2  662.37  4625.7  662.53
  4716.6  662.65  4736.7  661.78  4960.2  663.78  4970.4  664.86  4971.4  661.78
  4975.0  653.78  5025.0  653.78  5028.6  661.78  5043.0  663.64  5080.0  662.55
  5330.2  663.74  5427.1  666.86  5460.4  669.30  5490.1  674.87  5510.9  677.44
  5531.9  684.38  5569.2  693.46  5630.0  704.77  5731.2  715.56  5815.0  722.90
#Mann=5,-1,0
  4118.0    0.14       0  4625.7    0.08       0  4971.4   0.045       0
  5028.6    0.08       0  5731.2     0.1       0
Bank Sta=4971.4,5028.6
XS Rating Curve= 0
Exp/Cntr=0.3,0.1

Type RM Length L Ch R = 1,67698,386,386,386
BEGIN DESCRIPTION:
Dutchman Creek 71.0
END DESCRIPTION:
XS GIS Cut Line= 3
      1552059.87       797778.04      1551756.02       797443.80
      1551573.72       796866.51
#Sta/Elev= 30
  4214.1  697.42  4249.0  695.66  4302.2  695.18  4316.0  693.40  4325.9  693.90
  4360.3  686.07  4400.0  684.24  4418.6  681.69  4426.0  679.71  4461.3  675.06
  4557.5  667.26  4791.6  661.44  4815.0  662.16  4889.3  662.14  4937.3  663.40
  4967.0  663.03  4971.4  661.39  4975.0  653.39  5025.0  653.39  5028.6  661.39
  5029.5  665.17  5038.6  670.79  5051.3  676.27  5061.8  682.13  5074.6  686.53
  5085.0  689.64  5092.2  690.04  5128.7  695.41  5145.9  696.65  5271.2  704.77
#Mann=5,-1,0
  4214.1    0.06       0  4937.3    0.14       0  4971.4   0.045       0
  5028.6    0.14       0  5145.9    0.06       0
Bank Sta=4971.4,5028.6
XS Rating Curve= 0
Exp/Cntr=0.3,0.1

Type RM Length L Ch R = 1,67312,782,782,782
BEGIN DESCRIPTION:
Dutchman Creek 70.0
END DESCRIPTION:
XS GIS Cut Line= 5
      1552348.43       797666.06      1552254.18       797306.70
      1551947.82       796882.51      1551841.77       796776.46
      1551423.48       796623.28
#Sta/Elev= 30
  4114.0  720.52  4132.2  719.93  4201.4  707.25  4225.5  704.36  4308.5  689.01
  4320.4  687.74  4400.7  674.56  4431.6  668.43  4469.1  664.34  4539.3  661.64
  4577.0  661.96  4595.2  661.26  4738.2  661.32  4761.3  662.33  4885.6  662.84
  4915.4  662.89  4927.7  661.82  4960.6  662.32  4971.4  661.15  4975.0  653.15
  5025.0  653.15  5028.6  661.15  5043.0  669.31  5055.1  677.28  5060.2  678.81
  5154.7  697.06  5232.5  704.76  5273.6  706.97  5467.7  713.77  5604.2  716.89
#Mann=5,-1,0
  4114.0    0.06       0  4885.6    0.14       0  4971.4   0.045       0
  5028.6    0.14       0  5060.2    0.06       0
Bank Sta=4971.4,5028.6
XS Rating Curve= 0
Exp/Cntr=0.3,0.1

Type RM Length L Ch R = 1,66530,1013,1013,1013
BEGIN DESCRIPTION:
Dutchman Creek 69.0
END DESCRIPTION:
XS GIS Cut Line= 5
      1552767.30       797313.58      1552749.94       797105.26
      1552741.26       796753.70      1552611.05       796523.67
      1552524.25       796007.15
#Sta/Elev= 30
  4254.4  717.38  4260.5  716.10  4290.6  713.03  4359.2  698.66  4379.7  695.11
  4514.1  662.20  4535.1  661.38  4582.0  660.85  4678.7  661.40  4726.7  660.93
  4758.3  661.61  4788.1  660.60  4804.5  661.98  4831.4  661.55  4893.2  662.19
  4967.6  662.44  4971.4  660.60  4975.0  652.60  5025.0  652.60  5028.6  660.60
  5037.6  662.56  5113.3  661.50  5129.9  662.30  5164.9  664.84  5302.8  671.77
  5367.3  676.73  5499.3  683.88  5524.1  686.55  5585.9  688.86  5603.2  690.22
#Mann=4,-1,0
  4254.4    0.06       0  4893.2    0.14       0  4971.4   0.045       0
  5028.6    0.06       0
Bank Sta=4971.4,5028.6
XS Rating Curve= 0
Exp/Cntr=0.3,0.1

Type RM Length L Ch R = 1,65517,707,707,707
BEGIN DESCRIPTION:
Dutchman Creek 68.0
END DESCRIPTION:
XS GIS Cut Line= 3
      1553231.59       797181.09      1553302.28       796920.33
      1553570.00       796430.14
#Sta/Elev= 30
  4441.5  698.90  4457.4  696.83  4468.4  695.92  4479.0  696.41  4489.5  694.21
  4501.7  692.45  4553.1  685.94  4609.7  679.43  4650.4  675.44  4699.0  669.84
  4720.6  668.55  4749.1  665.64  4763.1  663.11  4796.7  661.53  4841.3  661.59
  4871.8  660.91  4962.7  661.18  4970.7  660.22  4971.4  659.70  4975.0  651.70
  5025.0  651.70  5028.6  659.70  5036.5  664.23  5072.3  676.39  5097.4  682.88
  5110.4  685.41  5159.3  692.99  5206.9  698.20  5234.5  700.25  5270.2  701.08
#Mann=4,-1,0
  4441.5    0.06       0  4501.7    0.14       0  4971.4   0.045       0
  5028.6    0.14       0
Bank Sta=4971.4,5028.6
XS Rating Curve= 0
Exp/Cntr=0.3,0.1

Type RM Length L Ch R = 1,64810,262,262,262
BEGIN DESCRIPTION:
Dutchman Creek 67.0
END DESCRIPTION:
XS GIS Cut Line= 5
      1554207.61       796785.44      1554159.34       796667.78
      1554029.63       796562.20      1553875.79       796450.59
      1553622.42       796426.46
#Sta/Elev= 30
  4710.6  710.34  4726.7  709.15  4743.8  706.16  4755.5  704.33  4796.0  694.43
  4808.6  688.40  4815.1  684.19  4820.9  679.38  4822.7  678.79  4832.5  679.06
  4875.9  676.88  4897.5  667.58  4916.9  663.15  4939.0  661.33  4971.7  660.07
  4975.3  651.07  5024.7  651.07  5028.3  660.07  5064.8  662.22  5128.7  663.65
  5183.8  666.05  5196.9  669.33  5205.5  670.43  5229.0  675.09  5248.8  676.88
  5260.0  679.91  5292.2  683.64  5361.3  694.21  5403.1  698.51  5449.6  700.71
#Mann=4,-1,0
  4710.6    0.12       0  4743.8    0.14       0  4971.7   0.045       0
  5028.3    0.14       0
Bank Sta=4971.7,5028.3
XS Rating Curve= 0
Exp/Cntr=0.5,0.3

Type RM Length L Ch R = 1,64548,112,112,112
BEGIN DESCRIPTION:
Milling Rd (DC) us
END DESCRIPTION:
XS GIS Cut Line= 6
      1554457.98       796417.41      1554180.45       796342.00
      1553830.54       796272.62      1553543.98       796148.94
      1553455.21       796046.40      1553431.88       795939.37
#Sta/Elev= 30
  4594.1  709.14  4607.7  708.65  4632.1  703.86  4776.5  699.16  4838.0  695.30
  4873.8  690.63  4921.6  676.84  4945.5  665.97  4969.9  660.03  4970.5  661.80
  4984.0  650.40  5016.0  650.40  5029.5  661.80  5112.6  662.46  5235.6  673.20
  5344.2  674.06  5363.2  675.67  5394.0  673.46  5453.5  672.91  5460.4  674.84
  5481.6  671.67  5636.9  664.30  5660.6  667.13  5682.3  666.60  5697.5  672.21
  5711.5  670.66  5729.3  677.45  5737.9  676.54  5765.6  687.16  5795.7  690.60
#Mann=4,-1,0
  4594.1    0.06       0  4776.5    0.14       0  4970.5   0.045       0
  5029.5    0.14       0
#XS Ineff=2,0
    0.00 4840.00  689.92 5160.00    0.00  676.13
Permanent Ineff=
       F       F
Bank Sta=4970.5,5029.5
XS Rating Curve= 0
Exp/Cntr=0.5,0.3

Type RM Length L Ch R =3,64493,,,
BEGIN DESCRIPTION:
Milling Rd (DC) tor
Structure ID: LDS_DC_05
Approximate Survey Structure
END DESCRIPTION:
Bridge Culvert--1,0,-1,-1,0
Deck Dist Width WeirC Skew NumUp NumDn MinLoCord MaxHiCord MaxSubmerge Is_Ogee
39.5,31,3,,13,13,,,0.95,0,1,1,,,
  4879.5  4879.5  5120.5  5120.5  5130.5  5272.0  5356.2  5408.1  5487.0  5632.8
  5680.0  5748.6  5808.5
  681.10  681.10  677.60  677.60  677.37  676.06  676.35  677.04  679.65  685.23
  687.85  692.00  696.58
  630.40  678.60  675.10  630.40  630.40  630.40  630.40  630.40  630.40  630.40
  630.40  630.40  630.40
  4879.5  4879.5  5120.5  5120.5  5130.5  5272.0  5356.2  5408.1  5487.0  5632.8
  5680.0  5748.6  5808.5
  681.10  681.10  677.60  677.60  677.37  676.06  676.35  677.04  679.65  685.23
  687.85  692.00  696.58
  630.40  678.60  675.10  630.40  630.40  630.40  630.40  630.40  630.40  630.40
  630.40  630.40  630.40
Pier Skew, UpSta & Num, DnSta & Num=,4903.6,2,4903.6,2,0,0,0,0,0
       3       3
  681.64  678.60
       3       3
  677.16  678.60
Pier Skew, UpSta & Num, DnSta & Num=,4951.8,2,4951.8,2,0,0,0,0,0
       3       3
  664.64  678.60
       3       3
  663.09  678.60
Pier Skew, UpSta & Num, DnSta & Num=,5000,2,5000,2,0,0,0,0,0
       3       3
  650.40  678.60
       3       3
  650.15  678.60
Pier Skew, UpSta & Num, DnSta & Num=,5048.2,2,5048.2,2,0,0,0,0,0
       3       3
  661.46  678.60
       3       3
  661.38  678.60
Pier Skew, UpSta & Num, DnSta & Num=,5096.4,2,5096.4,2,0,0,0,0,0
       3       3
  661.94  676.00
       3       3
  661.82  676.00
Abutment Skew #Up #Dn=,2,2
  4879.5  4892.0
  678.60  685.10
  4879.5  4892.0
  678.60  675.10
Abutment Skew #Up #Dn=,2,2
  5108.0  5120.5
  662.29  675.10
  5108.0  5120.5
  662.68  675.10
BR Coef=1,1,0,1.25,0,,,0.8,0,2,0,
WSPro=,,,, 1 ,,,, 0 ,,,, 0 ,,,,-1 ,-1 ,-1 , 0 , 0 , 0 , 0 , 0
BC Design=,,0,,0,,,,,,

Type RM Length L Ch R = 1,64436,517,517,517
BEGIN DESCRIPTION:
Milling Rd (DC) ds
END DESCRIPTION:
XS GIS Cut Line= 5
      1554494.14       796378.18      1554280.00       796263.57
      1553767.20       796142.91      1553616.37       796061.47
      1553444.44       795928.75
#Sta/Elev= 30
  4516.7  709.66  4672.7  697.35  4701.1  697.80  4819.0  689.66  4865.1  686.42
  4891.6  681.34  4919.5  672.63  4941.3  664.31  4964.4  661.00  4970.5  658.91
  4984.0  650.15  5016.0  650.15  5029.5  659.66  5044.9  661.49  5074.6  661.13
  5113.0  663.01  5216.3  663.55  5397.5  667.55  5485.6  664.43  5502.2  666.41
  5506.7  665.97  5512.5  667.43  5524.6  667.76  5535.4  672.18  5548.6  671.33
  5559.1  673.65  5580.9  681.64  5603.1  681.65  5612.2  684.63  5675.0  690.53
#Mann=4,-1,0
  4516.7    0.06       0  4819.0    0.14       0  4970.5   0.045       0
  5029.5    0.14       0
#XS Ineff=2,0
    0.00 4838.00  690.03 5162.00    0.00  675.98
Permanent Ineff=
       F       F
Bank Sta=4970.5,5029.5
XS Rating Curve= 0
Exp/Cntr=0.5,0.3

Type RM Length L Ch R = 1,63919,697,697,697
BEGIN DESCRIPTION:
Dutchman Creek 66.0
END DESCRIPTION:
XS GIS Cut Line= 3
      1554262.79       795810.78      1554101.03       795710.64
      1553461.79       795687.54
#Sta/Elev= 30
  4641.7  690.05  4669.4  689.30  4685.3  687.27  4699.4  683.50  4710.1  682.95
  4738.5  681.95  4756.7  679.54  4821.4  666.96  4860.3  661.73  4907.1  662.07
  4933.5  663.86  4944.9  663.83  4967.2  659.92  4968.1  659.03  4972.2  650.03
  5027.8  650.03  5031.9  659.03  5067.2  661.69  5096.2  660.06  5115.1  660.09
  5166.5  662.70  5198.9  662.46  5222.6  664.87  5234.0  667.02  5257.7  674.82
  5283.9  685.14  5328.2  697.19  5344.8  701.11  5411.0  713.21  5471.6  718.88
#Mann=4,-1,0
  4641.7    0.12       0  4710.1    0.06       0  4968.1   0.045       0
  5031.9    0.14       0
Bank Sta=4968.1,5031.9
XS Rating Curve= 0
Exp/Cntr=0.3,0.1

Type RM Length L Ch R = 1,63222,926,926,926
BEGIN DESCRIPTION:
Dutchman Creek 65.0
END DESCRIPTION:
XS GIS Cut Line= 4
      1554293.56       795803.07      1554162.64       795641.33
      1554178.04       795310.17      1554131.84       795094.57
#Sta/Elev= 30
  4527.6  690.69  4538.4  690.77  4584.2  686.05  4607.9  680.87  4671.9  669.52
  4713.1  665.65  4752.7  662.89  4820.2  661.76  4837.5  660.75  4858.2  661.85
  4894.1  661.85  4927.9  662.83  4938.4  662.23  4949.4  662.62  4964.0  661.32
  4968.1  658.86  4972.2  649.86  5027.8  649.86  5031.9  658.86  5043.8  659.78
  5094.2  667.61  5111.9  674.09  5121.4  678.46  5154.9  691.66  5198.9  706.30
  5221.7  711.65  5236.4  713.46  5257.6  714.63  5272.0  714.94  5287.7  713.96
#Mann=4,-1,0
  4527.6    0.12       0  4607.9    0.06       0  4968.1   0.045       0
  5031.9    0.14       0
Bank Sta=4968.1,5031.9
XS Rating Curve= 0
Exp/Cntr=0.3,0.1

Type RM Length L Ch R = 1,62296,1071,1071,1071
BEGIN DESCRIPTION:
Dutchman Creek 64.0
END DESCRIPTION:
XS GIS Cut Line= 4
      1555167.28       795993.82      1555130.39       795710.98
      1555011.52       795436.37      1554204.07       795120.77
#Sta/Elev= 30
  4564.8  705.89  4596.7  702.42  4633.1  700.30  4689.9  686.38  4753.5  666.99
  4780.8  660.64  4790.0  659.60  4840.0  660.40  4904.2  659.59  4958.5  662.86
  4964.0  660.51  4964.6  658.64  4969.1  649.64  5030.9  649.64  5035.4  658.64
  5054.5  658.72  5059.6  660.17  5085.1  661.99  5146.5  661.45  5323.3  660.93
  5449.6  663.34  5507.4  662.18  5562.7  663.16  5830.2  662.49  5865.2  662.88
  5892.7  666.47  5905.9  669.46  5971.6  697.16  5992.4  703.13  6016.2  708.12
#Mann=5,-1,0
  4564.8    0.12       0  4964.6   0.045       0  5035.4    0.12       0
  5146.5    0.06       0  5830.2    0.14       0
Bank Sta=4964.6,5035.4
XS Rating Curve= 0
Exp/Cntr=0.3,0.1

Type RM Length L Ch R = 1,61225,778,778,778
BEGIN DESCRIPTION:
Dutchman Creek 63.0
END DESCRIPTION:
XS GIS Cut Line= 4
      1556272.79       795564.30      1555980.17       795317.87
      1554278.16       794724.87      1553977.81       794486.12
#Sta/Elev= 30
  4557.2  706.99  4608.1  705.77  4688.4  699.72  4751.5  693.21  4795.3  687.63
  4930.0  666.02  4954.6  663.92  4961.2  661.90  4962.0  658.12  4964.6  658.27
  4969.1  649.27  5030.9  649.27  5035.4  658.27  5047.8  658.12  5061.2  661.77
  5315.6  661.40  5382.6  660.06  5581.0  660.99  5633.4  659.49  5765.8  659.03
  6280.9  661.41  6412.1  659.36  6593.9  661.09  6720.6  665.06  6791.7  667.04
  6830.5  672.44  6937.0  701.00  6959.6  704.13  7057.0  712.55  7125.8  716.02
#Mann=4,-1,0
  4557.2    0.12       0  4964.6   0.045       0  5035.4    0.12       0
  6720.6     0.1       0
#XS Ineff=2,0
       0                 6348.50    0.00  691.62
Permanent Ineff=
       F       F
Bank Sta=4964.6,5035.4
XS Rating Curve= 0
Exp/Cntr=0.3,0.1

Type RM Length L Ch R = 1,60447,729,729,729
BEGIN DESCRIPTION:
Dutchman Creek 62.0
END DESCRIPTION:
XS GIS Cut Line= 4
      1556701.53       794669.36      1556490.32       794569.32
      1554355.77       794480.38      1554055.60       794502.61
#Sta/Elev= 30
  4192.9  694.73  4279.7  688.46  4452.3  665.54  4494.8  662.51  4633.8  659.58
  4824.4  660.03  4954.8  662.48  4956.6  661.99  4957.4  657.94  4961.1  658.01
  4966.0  649.01  5034.0  649.01  5038.9  658.01  5051.7  657.94  5053.5  661.24
  5078.0  660.82  5435.8  661.38  5700.1  657.85  5795.4  659.47  6035.2  658.28
  6196.1  660.30  6290.4  658.36  6324.4  659.79  6543.2  660.16  6658.5  662.93
  6701.7  668.14  6744.4  678.79  6789.9  695.64  6829.9  708.05  6864.0  714.09
#Mann=5,-1,0
  4192.9     0.1       0  4961.1   0.045       0  5038.9     0.1       0
  5078.0    0.06       0  6543.2     0.1       0
#XS Ineff=2,0
       0                 6032.90    0.00  692.12
Permanent Ineff=
       F       F
Bank Sta=4961.1,5038.9
XS Rating Curve= 0
Exp/Cntr=0.3,0.1

Type RM Length L Ch R = 1,59718,1354,1354,1354
BEGIN DESCRIPTION:
Dutchman Creek 61.0
END DESCRIPTION:
XS GIS Cut Line= 5
      1556811.92       794592.42      1556671.81       794147.16
      1556075.28       793892.15      1555155.43       793764.64
      1554854.86       793227.28
#Sta/Elev= 30
  3573.4  697.52  3660.7  694.15  3871.2  680.86  3977.7  679.04  4023.4  676.57
  4041.3  675.38  4110.0  666.05  4139.0  664.43  4179.6  659.31  4503.1  660.91
  4638.3  659.70  4735.1  661.52  4862.4  661.75  4908.0  660.69  4939.6  661.47
  4964.6  657.76  4969.1  648.76  5030.9  648.76  5035.4  657.76  5036.5  662.22
  5058.7  660.47  5231.1  659.06  5545.5  658.76  5615.2  660.17  5760.9  659.81
  5878.5  663.14  5972.2  667.88  6067.6  678.39  6201.4  697.51  6233.3  704.15
#Mann=4,-1,0
  3573.4     0.1       0  4964.6   0.045       0  5035.4     0.1       0
  5615.2     0.1       0
#XS Ineff=2,0
       0                 5616.90    0.00  686.61
Permanent Ineff=
       F       F
Bank Sta=4964.6,5035.4
XS Rating Curve= 0
Exp/Cntr=0.3,0.1

Type RM Length L Ch R = 1,58364,1536,1536,1536
BEGIN DESCRIPTION:
Dutchman Creek 60.0
END DESCRIPTION:
XS GIS Cut Line= 6
      1557837.55       793304.71      1557359.42       792967.75
      1557040.66       792926.76      1556066.17       792676.31
      1555273.82       792548.80      1554977.83       792612.56
#Sta/Elev= 30
  3162.4  691.31  3275.3  684.50  3363.6  677.30  3602.0  667.56  3675.9  666.82
  3782.2  668.82  3825.6  670.04  3924.4  676.03  4052.7  680.26  4096.3  680.11
  4120.4  678.82  4218.4  663.76  4282.8  658.84  4796.9  659.82  4907.8  658.83
  4951.8  660.24  4963.5  657.26  4968.0  648.26  5032.0  648.26  5036.5  657.26
  5049.6  657.46  5053.8  659.99  5216.5  657.71  5657.1  658.96  5873.0  657.80
  5921.5  659.15  5989.2  663.43  6035.4  676.59  6094.8  685.03  6180.2  692.28
#Mann=3,-1,0
  3162.4     0.1       0  4963.5   0.045       0  5036.5     0.1       0
#XS Ineff=2,0
    0.00 4065.40  685.87 5669.20    0.00  685.87
Permanent Ineff=
       F       F
Bank Sta=4963.5,5036.5
XS Rating Curve= 0
Exp/Cntr=0.3,0.1
