--- Kerr Creek.prj (project) ---

Proj Title=.Kerr Creek Limited Detail Study
Current Plan=p01
Default Exp/Contr=0.3,0.1
English Units
Geom File=g01
Flow File=f01
Plan File=p01
Y Axis Title=Elevation
X Axis Title(PF)=Main Channel Distance
X Axis Title(XS)=Station
BEGIN DESCRIPTION:
Kerr Creek
END DESCRIPTION:
DSS Export Rating Curves= 0
DSS Export Rating Curve Sorted= 0
DSS Export Volume Flow Curves= 0
DXF OffsetX= 0
DXF OffsetY= 0
DXF ScaleX= 1
DXF ScaleY= 10

--- Kerr Creek.p01 (plan) ---

Plan Title=Floodway Run
Program Version=3.12
Short Identifier=Floodway
Geom File=g01
Flow File=f01
Subcritical Flow
K Sum by GR= 0
Std Step Tol= 0.01
Critical Tol= 0.01
Num of Std Step Trials= 20
Max Error Tol= 0.3
Flow Tol Ratio= 0.001
Split Flow NTrial= 30
Split Flow Tol= 0.02
Split Flow Ratio= 0.02
Log Output Level= 0
Friction Slope Method= 1
Unsteady Friction Slope Method= 2
Unsteady Bridges Friction Slope Method= 1
Parabolic Critical Depth
Global Vel Dist= 0 , 0 , 0
Global Log Level= 0
CheckData=True
Encroach Param=-1 ,10,10, 2
Encroach River=Kerr Creek
Encroach Reach=Reach-1
Encroach Node=39867
       1 4958.81    5010
Encroach Node=39712
       1 4983.14    5012
Encroach Node=39530
       1 4949.12    5012
Encroach Node=39331
       1    4992    5030
Encroach Node=38995
       1    4890    5051
Encroach Node=38887
       1  4860.2  5054.2
Encroach Node=38769
       1    4862    5022
Encroach Node=38630
       1    4988 5019.65
Encroach Node=38481
       1    4994    5011
Encroach Node=38224
       1    4996    5015
Encroach Node=37999
       1  4996.5    5012
Encroach Node=37696
       1    4980    5010
Encroach Node=37499
       1    4992    5008
Encroach Node=37366
       1    4995    5012
Encroach Node=37210
       1    4987    5018
Encroach Node=37142
       1    4984    5016
Encroach Node=37060
       1    4987    5019
Encroach Node=36929
       1    4990    5007
Encroach Node=36807
       1    4990    5018
Encroach Node=36504
       1    4988 5016.88
Encroach Node=36011
       1    4988    5012
Encroach Node=35783
       1    4994 5015.72
Encroach Node=35335
       1    4988    5012
Encroach Node=35000
       1    4995    5010
Encroach Node=34518
       1    4988    5011
Encroach Node=34175
       1 4984.03    5012
Encroach Node=33856
       1    4988 5017.44
Encroach Node=33480
       1    4970    5035
Encroach Node=33116
       1    4930    5050
Encroach Node=32503
       1    4915    5025
Encroach Node=32128
       1    4950    5050
Encroach Node=32025
       1    4958    5043
Encroach Node=31500
       1 4969.25 5068.93
Encroach Node=31013
       1    4970    5025
Encroach Node=30511
       1 4935.46    5023
Encroach Node=30004
       1 4928.44 5019.84
Encroach Node=29516
       1 4985.76 5135.56
Encroach Node=29013
       1  4984.1 5070.38
Encroach Node=28499
       1 4983.88 5103.39
Encroach Node=28014
       1    4960    5040
Encroach Node=27501
       1 4890.39 5042.72
Encroach Node=27003
       1 4935.42 5064.04
Encroach Node=26502
       1 4964.68 5097.57
Encroach Node=26275
       1  4982.5 5062.61
Encroach Node=26015
       1    4992    5035
Encroach Node=25700
       1    4941    5013
Encroach Node=25543
       1    4955    5043
Encroach Node=25215
       1    4976    5027
Encroach Node=25111
       1  4986.8  5013.2
Encroach Node=25041
       1    4990    5035
Encroach Node=24315
       1    4983    5022
Encroach Node=24001
       1 4976.87    5075
Encroach Node=23493
       1  4981.8 5075.14
Encroach Node=22993
       1  4981.8    5029
Encroach Node=22629
       1  4981.8 5054.67
Encroach Node=21999
       1  4981.8    5035
Encroach Node=21515
       1    4965    5065
Encroach Node=20996
       1 4946.19 5098.02
Encroach Node=20342
       1    4960    5035
Encroach Node=19998
       1    4950    5050
Encroach Node=19449
       1    4950    5045
Encroach Node=19335
       1    4975    5025
Encroach Node=18999
       1    4987    5030
Encroach Node=18490
       1    4975    5050
Encroach Node=18242
       1    4929    5080
Encroach Node=17793
       1    4840  5019.4
Encroach Node=17515
       1    4945    5065
Encroach Node=17000
       1 4900.48    5099
Encroach Node=16497
       1    4930    5104
Encroach Node=16177
       1 4958.28    5050
Encroach Node=15814
       1  4980.6    5045
Encroach Node=15498
       1    4920    5050
Encroach Node=15333
       1 4817.61 5069.49
Encroach Node=14994
       1    4802    5100
Encroach Node=14289
       1 4831.53    5020
Encroach Node=13998
       1 4844.98 5036.67
Encroach Node=13497
       1 4881.05  5191.5
Encroach Node=13307
       1 4928.72 5054.88
Encroach Node=13111
       1 4918.72 5064.88
Encroach Node=12726
       1    4840 5105.59
Encroach Node=12212
       1    4960    5060
Encroach Node=11764
       1 4876.59 5083.77
Encroach Node=11495
       1 4835.16    5020
Encroach Node=11137
       1 4808.14    5020
Encroach Node=10795
       1    4906    5094
Encroach Node=10627
       1 4870.28 5115.28
Encroach Node=10420
       1 4884.56 5066.13
Encroach Node=10000
       1 4845.78 5173.34
Encroach Node=9629
       1 4929.62    5100
Encroach Node=9137
       1  4880.7 5119.98
Encroach Node=8814
       1    4925    5055
Encroach Node=8700
       1    4860    5060
Encroach Node=8504
       1    4790    5230
Encroach Node=8264
       1    4880    5120
Encroach Node=7995
       1 4867.22 5063.21
Encroach Node=7519
       1  4778.1 5094.39
Encroach Node=6901
       1  4978.7 5185.91
Encroach Node=6226
       1 4947.81 5078.06
Encroach Node=5748
       1 4834.26 5089.57
Encroach Node=5330
       1 4811.34  5021.3
Encroach Node=5000
       1 4718.37 5065.64
Encroach Node=4493
       1 4807.31  5217.3
Encroach Node=4003
       1    4850    5050
Encroach Node=3674
       1    4942    5042
Encroach Node=3499
       1    4910    5050
Encroach Node=2815
       1    4750  5021.3
Encroach Node=2348
       1 4822.95  5021.3
Encroach Node=2024
       1 4753.55  5021.3
Encroach Node=1511
       1  4820.2 5223.53
Encroach Node=898
       1 4780.19  5021.3
Encroach Node=745
       1 4834.89  5021.3
BEGIN DESCRIPTION:
Floodway Run
END DESCRIPTION:
Computation Interval=1HOUR
Output Interval=1HOUR
Run HTab= 0
Run UNet= 0
Run PostProcess= 0
UNET Theta= 1
UNET Theta Warmup= 1
UNET ZTol= 0.02
UNET ZSATol= 0.05
UNET MxIter= 20
UNET MaxInSteps= 0
UNET DtIC= 0
UNET DtMin= 0
UNET MaxCRTS= 20
UNET WFStab= 2
UNET SFStab= 1
UNET WFX= 1
UNET SFX= 1
UNET DSS MLevel= 4
UNET DZMax Abort= 100
UNET Convert EG Bridges=-1
UNET Use Existing IB Tables=-1
UNET Froude Reduction=False
UNET Froude Limit= 1
UNET Froude Power= 10
Instantaneous Interval=1HOUR
Write IC File= 0
Echo Input=False
Echo Output=False
Write Detailed= 0
Detailed Automatic Start=False, 10

--- Kerr Creek.f01 (steady flow) ---

Flow Title=Floodway
Number of Profiles=2
Profile Names=100-year,100-FW
River Rch & RM= Kerr Creek,Reach-1,39867
     488     488
River Rch & RM= Kerr Creek,Reach-1,36504
     651     651
River Rch & RM= Kerr Creek,Reach-1,33856
     906     906
River Rch & RM= Kerr Creek,Reach-1,32503
    1202    1202
River Rch & RM= Kerr Creek,Reach-1,29013
    1823    1823
River Rch & RM= Kerr Creek,Reach-1,27003
    2230    2230
River Rch & RM= Kerr Creek,Reach-1,24315
    2486    2486
River Rch & RM= Kerr Creek,Reach-1,20996
    2713    2713
River Rch & RM= Kerr Creek,Reach-1,18490
    2919    2919
River Rch & RM= Kerr Creek,Reach-1,14289
    3123    3123
River Rch & RM= Kerr Creek,Reach-1,10000
    3314    3314
River Rch & RM= Kerr Creek,Reach-1,6901
    3509    3509
Boundary for River Rch & Prof#=Kerr Creek,Reach-1,1
Up Type=0
Dn Type=3
Dn Slope=0.0017
Boundary for River Rch & Prof#=Kerr Creek,Reach-1,2
Up Type=0
Dn Type=3
Dn Slope=0.0017

--- Kerr Creek.g01 (geometry) ---

Geom Title=Existing Conditions

River Reach=Kerr Creek,Reach-1
Reach XY= 30
      1498864.65       668249.24      1498730.48       668854.55
      1498936.63       670326.88      1499262.38       670794.63
      1499593.63       672064.13      1499448.88       673795.75
      1499087.00       674303.81      1498985.63       674889.50
      1499414.88       675585.50      1501866.75       677488.63
      1502325.00       679062.88      1502675.38       681224.69
      1502750.25       681356.44      1502965.88       681323.50
      1504118.50       682922.31      1504307.13       683548.06
      1504394.00       684952.25      1505289.13       685106.44
      1505567.63       685546.56      1506600.50       686212.69
      1507376.00       687104.94      1507879.00       688946.25
      1508929.88       690754.63      1510139.50       693489.63
      1510471.75       694679.75      1511777.13       696030.06
      1512648.50       697542.00      1514205.38       699314.50
      1515510.75       699739.63      1516712.60       700573.39

Type RM Length L Ch R = 1,39867,155,155,155
BEGIN DESCRIPTION:
Dam KC_11 (Kerr) ds
END DESCRIPTION:
XS GIS Cut Line= 4
      1498209.59       669199.00      1498714.32       669158.18
      1498768.13       669150.76      1499289.51       669007.89
#Sta/Elev= 30
  4442.1  893.15  4493.6  893.06  4588.5  884.35  4682.7  880.94  4718.8  877.60
  4766.8  875.12  4809.7  868.63  4823.7  864.86  4869.7  858.85  4879.4  858.83
  4893.7  856.80  4928.8  843.31  4965.7  842.15  4998.0  840.67  4999.0  838.67
  5001.0  838.67  5002.0  840.67  5002.8  842.64  5005.8  844.29  5023.2  846.84
  5060.5  857.06  5075.3  860.42  5145.2  869.41  5200.6  874.65  5243.6  877.64
  5261.8  880.19  5314.0  883.67  5352.8  889.15  5429.2  896.58  5543.4  900.49
#Mann=5,-1,0
  4442.1    0.09       0  4965.7    0.13       0  4998.0    0.05       0
  5002.0    0.13       0  5060.5    0.09       0
#XS Ineff=2,0
    0.00 4958.80  845.17 5012.00    0.00  845.34
Permanent Ineff=
       F       F
Bank Sta=4998,5002
XS Rating Curve= 0
Exp/Cntr=0.3,0.1

Type RM Length L Ch R = 1,39712,182,182,182
BEGIN DESCRIPTION:
Kerr Creek 84.0
END DESCRIPTION:
XS GIS Cut Line= 3
      1498396.60       669447.08      1498781.22       669304.58
      1499176.67       669141.29
#Sta/Elev= 30
  4588.5  889.22  4594.5  889.44  4606.8  889.68  4622.3  889.13  4690.2  884.38
  4704.7  882.29  4805.2  870.87  4841.8  865.87  4885.6  858.69  4900.2  855.04
  4908.0  854.12  4923.9  849.14  4963.7  840.82  4980.3  840.45  4998.0  839.30
  4999.0  837.30  5001.0  837.30  5002.0  839.30  5009.4  841.40  5035.4  844.58
  5105.9  857.02  5123.6  861.05  5178.5  868.79  5193.9  869.54  5260.0  875.10
  5279.0  877.27  5298.1  880.22  5332.1  882.42  5369.2  887.35  5426.5  891.54
#Mann=5,-1,0
  4588.5    0.09       0  4594.5    0.13       0  4998.0    0.05       0
  5002.0    0.13       0  5178.5    0.09       0
Bank Sta=4998,5002
XS Rating Curve= 0
Exp/Cntr=0.3,0.1

Type RM Length L Ch R = 1,39530,199,199,199
BEGIN DESCRIPTION:
Kerr Creek 83.0
END DESCRIPTION:
XS GIS Cut Line= 3
      1498527.68       669559.01      1498840.56       669472.34
      1499140.80       669362.39
#Sta/Elev= 30
  4672.2  882.68  4715.1  880.96  4736.0  880.76  4741.9  880.20  4796.5  872.45
  4850.5  861.43  4866.5  857.07  4891.6  847.51  4901.0  843.35  4913.9  839.20
  4935.9  838.45  4996.7  838.66  4998.0  837.92  4999.0  835.92  5001.0  835.92
  5002.0  837.92  5015.7  841.74  5024.1  843.53  5043.1  848.84  5053.5  850.37
  5058.8  851.59  5069.0  852.95  5081.4  855.28  5117.6  860.11  5202.7  867.91
  5216.9  868.54  5272.6  872.74  5295.9  873.64  5306.0  874.66  5316.6  875.00
#Mann=3,-1,0
  4672.2    0.13       0  4998.0    0.05       0  5002.0    0.13       0
Bank Sta=4998,5002
XS Rating Curve= 0
Exp/Cntr=0.3,0.1

Type RM Length L Ch R = 1,39331,336,336,336
BEGIN DESCRIPTION:
Kerr Creek 82.0
END DESCRIPTION:
XS GIS Cut Line= 3
      1498518.29       669665.49      1498838.44       669647.82
      1499135.79       669690.30
#Sta/Elev= 30
  4677.7  879.35  4698.0  878.40  4719.4  878.47  4799.0  874.69  4812.9  873.03
  4833.1  871.27  4887.9  863.48  4900.1  861.25  4912.2  858.61  4930.3  855.70
  4949.3  850.37  4998.0  835.76  4999.0  833.76  5001.0  833.76  5002.0  835.76
  5049.2  836.16  5064.8  837.00  5085.1  839.30  5103.5  842.33  5116.8  845.27
  5141.8  849.43  5159.4  851.53  5173.8  854.36  5183.3  855.51  5231.4  865.31
  5243.5  868.51  5259.4  871.94  5278.7  874.61  5294.8  876.51  5298.7  876.73
#Mann=3,-1,0
  4677.7    0.13       0  4998.0    0.05       0  5002.0    0.13       0
Bank Sta=4998,5002
XS Rating Curve= 0
Exp/Cntr=0.3,0.1

Type RM Length L Ch R = 1,38995,108,108,108
BEGIN DESCRIPTION:
Kerr Creek 81.0
END DESCRIPTION:
XS GIS Cut Line= 5
      1498652.37       669816.96      1498813.07       669979.77
      1498903.98       669975.54      1498958.96       669969.20
      1499240.16       669791.60
#Sta/Elev= 30
  4676.0  864.72  4726.6  861.65  4772.2  857.81  4785.8  855.83  4800.4  853.03
  4810.1  851.75  4856.6  843.23  4879.9  839.94  4885.8  836.91  4896.8  829.86
  4999.0  827.86  5045.6  829.86  5046.3  831.66  5051.1  834.29  5059.9  837.14
  5089.0  843.79  5103.3  845.47  5132.2  851.15  5161.7  855.88  5183.0  857.80
  5189.7  859.30  5211.7  861.53  5218.6  862.97  5244.1  865.61  5274.5  867.75
  5288.7  869.72  5302.4  871.14  5335.4  873.65  5366.6  875.33  5383.7  875.88
#Mann=3,-1,0
  4676.0    0.13       0  4896.8   0.035       0  5045.6    0.13       0
Bank Sta=4896.8,5045.6
XS Rating Curve= 0
Exp/Cntr=0.3,0.1

Type RM Length L Ch R = 1,38887,118,118,118
BEGIN DESCRIPTION:
Kerr Creek 80.0
END DESCRIPTION:
XS GIS Cut Line= 3
      1498547.94       670170.53      1498932.84       670080.14
      1499215.65       670030.57
#Sta/Elev= 30
  4602.8  858.48  4607.8  858.13  4620.8  858.36  4641.1  857.88  4685.4  855.33
  4710.5  852.96  4752.8  848.43  4781.7  845.13  4800.6  842.39  4843.0  837.65
  4859.2  836.25  4860.2  833.86  4862.5  826.37  4999.0  824.37  5052.6  826.37
  5054.2  833.96  5055.2  834.97  5071.1  838.35  5087.7  840.48  5101.7  845.85
  5116.0  849.60  5127.5  851.82  5134.2  853.60  5164.5  860.23  5174.4  862.15
  5223.6  869.71  5242.2  871.68  5250.1  872.79  5275.4  874.73  5285.3  875.13
#Mann=3,-1,0
  4602.8    0.13       0  4862.5   0.035       0  5052.6    0.13       0
Bank Sta=4862.5,5052.6
XS Rating Curve= 0
Exp/Cntr=0.5,0.3

Type RM Length L Ch R = 1,38769,139,139,139
BEGIN DESCRIPTION:
Dam KC_10 (Kerr) us
END DESCRIPTION:
XS GIS Cut Line= 3
      1498508.48       670244.00      1498983.95       670187.25
      1499318.70       670208.87
#Sta/Elev= 30
  4520.7  860.91  4536.5  860.33  4548.0  860.30  4618.2  856.74  4666.2  854.75
  4682.3  854.54  4736.7  851.39  4777.4  845.36  4825.4  837.36  4835.6  836.86
  4857.9  826.77  4863.3  822.77  4999.0  820.77  5020.9  822.77  5024.1  826.79
  5037.8  835.59  5046.4  836.59  5056.9  839.47  5067.6  843.43  5117.1  859.78
  5127.2  862.68  5161.9  870.91  5188.2  876.31  5200.0  877.43  5217.5  879.84
  5230.7  880.66  5240.8  882.09  5273.4  884.70  5307.8  886.05  5335.0  886.61
#Mann=3,-1,0
  4520.7    0.13       0  4863.3   0.035       0  5020.9    0.13       0
#XS Ineff=2,0
    0.00 4862.00  832.79 5022.00    0.00  832.97
Permanent Ineff=
       F       F
Bank Sta=4863.3,5020.9
XS Rating Curve= 0
Exp/Cntr=0.5,0.3

Type RM Length L Ch R =5,38727,,,
BEGIN DESCRIPTION:
Dam KC_10 TOR (Kerr)
Structure ID: KC_10
Approximate Survey Structure
END DESCRIPTION:
#Inline Weir SE= 22
  4517.9  861.13  4553.6  859.67  4590.4  858.01  4637.2  855.94  4692.8  853.88
  4742.8  849.92  4775.7  845.43  4800.2  841.42  4833.0  837.24  4888.0  835.88
  4959.3  834.35  5025.0  834.34  5034.7  837.21  5068.1  847.59  5087.7  854.32
  5118.0  863.75  5152.1  871.97  5164.8  874.51  5197.9  879.57  5230.3  882.83
  5271.3  885.54  5296.7  886.47
IW Dist,WD,Coef,Skew,MaxSub,Min_El,Is_Ogee,SpillHt,DesHd
25,34,3,,0.95,,0,,,1,1

Type RM Length L Ch R = 1,38630,149,149,149
BEGIN DESCRIPTION:
Dam KC_10 (Kerr) ds
END DESCRIPTION:
XS GIS Cut Line= 3
      1498565.82       670366.31      1498936.32       670292.97
      1499285.73       670233.02
#Sta/Elev= 30
  4622.0  860.84  4713.1  857.03  4752.3  856.09  4794.8  850.30  4845.7  845.54
  4875.0  840.29  4898.4  837.19  4932.5  830.46  4965.1  827.82  4980.8  827.16
  4997.7  821.42  4998.0  820.11  4999.0  818.11  5001.0  818.11  5002.0  820.11
  5003.5  821.10  5015.9  823.31  5035.5  824.53  5046.0  826.94  5067.8  829.59
  5089.3  834.40  5114.9  841.01  5149.6  852.70  5179.4  861.91  5210.3  870.08
  5226.4  873.52  5270.1  880.67  5282.9  882.05  5305.0  884.01  5354.2  886.67
#Mann=4,-1,0
  4622.0    0.09       0  4845.7    0.13       0  4998.0    0.05       0
  5002.0    0.13       0
#XS Ineff=2,0
    0.00 4988.00  826.38 5019.70    0.00  826.32
Permanent Ineff=
       F       F
Bank Sta=4998,5002
XS Rating Curve= 0
Exp/Cntr=0.5,0.3

Type RM Length L Ch R = 1,38481,257,257,257
BEGIN DESCRIPTION:
Kerr Creek 79.0
END DESCRIPTION:
XS GIS Cut Line= 3
      1498728.76       670613.69      1499017.39       670403.77
      1499297.28       670237.59
#Sta/Elev= 30
  4643.2  855.76  4742.0  851.62  4804.8  845.83  4820.7  843.83  4835.1  839.74
  4859.0  837.16  4878.6  836.09  4904.4  835.84  4936.3  830.40  4943.9  828.46
  4986.1  826.12  4998.0  819.80  4999.0  817.80  5001.0  817.80  5002.0  819.80
  5002.6  820.01  5015.7  824.42  5041.3  827.07  5050.5  831.28  5080.4  843.35
  5094.1  850.07  5111.6  856.04  5124.2  859.82  5149.3  866.16  5161.2  868.04
  5186.5  874.26  5219.6  880.07  5248.7  883.32  5320.6  887.37  5325.6  887.16
#Mann=4,-1,0
  4643.2    0.09       0  4998.0    0.05       0  5002.0    0.09       0
  5002.6    0.13       0
Bank Sta=4998,5002
XS Rating Curve= 0
Exp/Cntr=0.3,0.1

Type RM Length L Ch R = 1,38224,225,225,225
BEGIN DESCRIPTION:
Kerr Creek 78.5
END DESCRIPTION:
XS GIS Cut Line= 2
      1499041.02       670703.13      1499265.04       670518.81
#Sta/Elev= 30
  4856.9  840.22  4865.4  838.69  4874.1  837.72  4883.5  836.38  4895.2  833.39
  4898.4  832.90  4908.6  831.98  4914.9  830.74  4941.9  827.20  4953.6  826.50
  4967.9  825.94  4974.4  825.85  4990.6  826.25  4995.0  823.03  4998.0  816.23
  4999.0  814.23  5001.0  814.23  5002.0  816.23  5007.2  820.32  5023.3  822.51
  5025.1  823.45  5039.4  822.94  5053.2  823.72  5066.9  824.26  5071.9  825.91
  5087.5  835.73  5103.4  842.08  5105.7  842.79  5132.8  849.26  5147.0  852.14
#Mann=4,-1,0
  4856.9    0.09       0  4874.1    0.13       0  4998.0    0.05       0
  5002.0    0.13       0
Bank Sta=4998,5002
XS Rating Curve= 0
Exp/Cntr=0.3,0.1

Type RM Length L Ch R = 1,37999,303,303,303
BEGIN DESCRIPTION:
Kerr Creek 78.0
END DESCRIPTION:
XS GIS Cut Line= 3
      1498960.27       670835.28      1499260.55       670800.30
      1499525.03       670775.00
#Sta/Elev= 30
  4694.2  852.18  4721.7  850.94  4745.2  848.78  4762.3  847.71  4795.7  843.76
  4822.4  841.91  4829.8  840.20  4857.0  835.13  4869.3  832.51  4894.5  825.94
  4905.3  823.77  4918.5  821.98  4938.6  820.22  4976.8  819.52  4994.6  818.35
  4996.5  816.84  4998.0  813.18  4999.0  811.18  5001.0  811.18  5002.0  813.18
  5003.6  814.78  5030.9  815.66  5057.8  820.46  5100.6  824.21  5114.3  824.87
  5159.0  828.48  5192.3  830.38  5201.9  832.23  5241.6  835.85  5262.2  838.95
#Mann=4,-1,0
  4694.2    0.09       0  4857.0    0.13       0  4998.0    0.05       0
  5002.0    0.13       0
Bank Sta=4998,5002
XS Rating Curve= 0
Exp/Cntr=0.3,0.1

Type RM Length L Ch R = 1,37696,197,197,197
BEGIN DESCRIPTION:
Kerr Creek 77.5
END DESCRIPTION:
XS GIS Cut Line= 3
      1499162.93       671128.70      1499296.20       671100.35
      1499503.15       671037.98
#Sta/Elev= 30
  4816.6  839.17  4819.6  838.60  4824.9  838.06  4837.3  836.41  4854.4  834.51
  4866.1  833.47  4869.8  832.79  4877.1  831.25  4881.4  830.63  4900.1  827.06
  4911.2  825.39  4951.0  818.79  4963.8  816.94  4974.6  816.55  4977.9  816.15
  4998.0  811.63  4999.0  809.63  5001.0  809.63  5002.0  811.63  5009.1  816.08
  5017.5  817.34  5037.0  818.04  5040.5  818.45  5052.1  820.08  5090.0  827.79
  5119.3  833.84  5138.1  838.42  5148.0  840.43  5159.6  841.75  5169.0  843.07
#Mann=4,-1,0
  4816.6    0.09       0  4998.0    0.05       0  5002.0    0.09       0
  5090.0    0.13       0
Bank Sta=4998,5002
XS Rating Curve= 0
Exp/Cntr=0.3,0.1

Type RM Length L Ch R = 1,37499,133,133,133
BEGIN DESCRIPTION:
Kerr Creek 77.0
END DESCRIPTION:
XS GIS Cut Line= 3
      1499161.43       671360.68      1499409.25       671270.30
      1499639.59       671112.85
#Sta/Elev= 30
  4737.5  841.25  4753.3  840.50  4778.0  838.60  4803.8  836.25  4830.2  834.30
  4864.0  831.38  4889.7  828.74  4900.0  827.47  4923.5  823.46  4936.2  820.65
  4947.7  818.56  4959.1  816.11  4976.9  813.55  4985.5  812.94  4998.0  809.72
  4999.0  807.72  5001.0  807.72  5002.0  809.72  5008.4  813.22  5011.8  814.12
  5032.0  817.38  5053.0  820.32  5067.2  823.05  5111.1  833.99  5140.8  839.15
  5194.7  847.77  5229.9  852.40  5248.4  855.13  5259.2  856.39  5280.3  857.29
#Mann=5,-1,0
  4737.5    0.09       0  4998.0    0.05       0  5002.0    0.09       0
  5032.0    0.13       0  5259.2    0.09       0
Bank Sta=4998,5002
XS Rating Curve= 0
Exp/Cntr=0.3,0.1

Type RM Length L Ch R = 1,37366,156,156,156
BEGIN DESCRIPTION:
Kerr Creek 76.0
END DESCRIPTION:
XS GIS Cut Line= 3
      1499170.37       671449.86      1499455.82       671392.77
      1499853.28       671293.40
#Sta/Elev= 30
  4708.1  842.62  4781.7  837.97  4861.0  832.05  4879.4  830.32  4901.9  827.09
  4917.1  824.03  4947.6  819.85  4983.3  813.89  4998.0  807.89  4999.0  805.89
  5001.0  805.89  5002.0  807.89  5009.8  808.67  5022.0  811.13  5044.6  814.79
  5064.1  818.87  5125.1  832.63  5153.1  837.67  5192.3  843.32  5220.1  846.52
  5234.5  846.60  5252.5  847.94  5280.7  848.87  5302.1  850.03  5313.0  850.80
  5329.9  852.72  5352.2  854.41  5365.9  854.54  5392.1  855.53  5408.9  856.93
#Mann=3,-1,0
  4708.1    0.09       0  4998.0    0.05       0  5002.0    0.09       0
Bank Sta=4998,5002
XS Rating Curve= 0
Exp/Cntr=0.3,0.1

Type RM Length L Ch R = 1,37210,68,68,68
BEGIN DESCRIPTION:
Kerr Creek 75.5
END DESCRIPTION:
XS GIS Cut Line= 3
      1499307.51       671534.15      1499503.17       671531.31
      1499681.80       671483.11
#Sta/Elev= 30
  4771.8  832.50  4781.1  831.44  4792.0  831.56  4813.8  826.07  4824.1  825.22
  4834.6  825.27  4849.6  824.62  4858.2  824.47  4877.9  822.45  4889.2  821.59
  4914.0  818.72  4920.0  817.75  4942.3  815.24  4946.8  815.04  4964.8  812.93
  4970.8  812.47  4983.3  810.74  4993.2  809.55  4995.7  808.53  4998.0  805.93
  4999.0  803.93  5001.0  803.93  5002.0  805.93  5029.5  813.60  5039.2  816.70
  5057.6  819.64  5109.3  831.65  5123.4  834.39  5146.8  838.27  5152.5  838.77
#Mann=3,-1,0
  4771.8    0.09       0  4998.0    0.05       0  5002.0    0.09       0
Bank Sta=4998,5002
XS Rating Curve= 0
Exp/Cntr=0.5,0.3

Type RM Length L Ch R = 1,37142,82,82,82
BEGIN DESCRIPTION:
Upright Avenue (Kerr) us
END DESCRIPTION:
XS GIS Cut Line= 5
      1499198.94       671549.66      1499512.64       671584.09
      1499542.76       671589.26      1499564.58       671591.01
      1499798.91       671573.70
#Sta/Elev= 30
  4653.3  844.72  4673.5  843.97  4688.2  842.33  4720.5  840.31  4738.3  838.45
  4750.2  835.86  4779.1  831.10  4792.6  830.41  4808.1  825.78  4823.3  825.01
  4837.1  825.34  4881.4  823.39  4892.2  822.76  4908.8  820.89  4960.2  812.46
  4994.0  803.40  4995.0  802.10  5005.0  802.10  5006.0  803.40  5008.7  806.32
  5038.1  810.42  5049.3  812.75  5073.0  816.54  5127.6  826.90  5140.1  828.50
  5154.8  830.98  5194.7  836.31  5225.9  838.61  5242.5  841.54  5256.3  842.92
#Mann=3,-1,0
  4653.3    0.09       0  4994.0    0.05       0  5006.0    0.09       0
#XS Ineff=2,0
    0.00 4953.60  808.90 5046.40    0.00  808.90
Permanent Ineff=
       F       F
Bank Sta=4994,5006
XS Rating Curve= 0
Exp/Cntr=0.5,0.3

Type RM Length L Ch R =3,37103,,,
BEGIN DESCRIPTION:
Upright Avenue TOR (Kerr)
Structure ID: LDS_KC_09
Approximate Survey Structure
END DESCRIPTION:
Bridge Culvert--1,0,-1,-1,0
Deck Dist Width WeirC Skew NumUp NumDn MinLoCord MaxHiCord MaxSubmerge Is_Ogee
34.5,9,3,,25,25,,,,0,1,1,,,
  4644.2  4671.6  4713.4  4734.8  4773.4  4789.2  4811.9  4828.4  4837.1  4865.3
  4903.8  4934.3  4951.7  4971.0  4983.5  4983.5  5016.5  5016.5  5061.5  5085.6
  5121.7  5159.3  5196.9  5240.9  5294.3
  844.78  843.28  840.16  837.42  829.10  828.63  823.99  824.38  824.38  823.11
  820.80  816.18  812.82  810.27  808.90  808.90  808.90  808.90  809.08  813.17
  818.78  825.36  830.87  837.07  842.61
  782.10  782.10  782.10  782.10  782.10  782.10  782.10  782.10  782.10  782.10
  782.10  782.10  782.10  782.10  782.10  807.90  807.90  782.10  782.10  782.10
  782.10  782.10  782.10  782.10  782.10
  4644.2  4671.6  4713.4  4734.8  4773.4  4789.2  4811.9  4828.4  4837.1  4865.3
  4903.8  4934.3  4951.7  4971.0  4983.5  4983.5  5016.5  5016.5  5061.5  5085.6
  5121.7  5159.3  5196.9  5240.9  5294.3
  844.78  843.28  840.16  837.42  829.10  828.63  823.99  824.38  824.38  823.11
  820.80  816.18  812.82  810.27  808.90  808.90  808.90  808.90  809.08  813.17
  818.78  825.36  830.87  837.07  842.61
  782.10  782.10  782.10  782.10  782.10  782.10  782.10  782.10  782.10  782.10
  782.10  782.10  782.10  782.10  782.10  807.90  807.90  782.10  782.10  782.10
  782.10  782.10  782.10  782.10  782.10
Pier Skew, UpSta & Num, DnSta & Num=,4991.8,2,4991.8,2,0,0,0,0,0
       1       1
  804.00  807.90
       1       1
  803.00  807.90
Pier Skew, UpSta & Num, DnSta & Num=,5008.3,2,5008.3,2,0,0,0,0,0
       1       1
  805.50  807.90
       1       1
  803.00  807.90
BR Coef=1,1,0,1.25,0,,,0.8,0,2,0,
WSPro=,,,, 1 ,,,, 0 ,,,, 0 ,,,,-1 ,-1 ,-1 , 0 , 0 , 0 , 0 , 0
BC Design=,,0,,0,,,,,,

Type RM Length L Ch R = 1,37060,131,131,131
BEGIN DESCRIPTION:
Upright Avenue (Kerr) ds
END DESCRIPTION:
XS GIS Cut Line= 5
      1499180.33       671612.18      1499458.73       671635.87
      1499525.87       671669.74      1499578.16       671694.17
      1499800.50       671619.70
#Sta/Elev= 30
  4648.8  844.68  4700.2  841.85  4726.5  838.67  4752.7  836.85  4761.0  834.60
  4776.7  832.26  4806.4  825.52  4813.1  824.78  4818.0  824.37  4841.6  823.64
  4877.6  820.78  4924.7  818.94  4942.2  815.92  4994.0  802.61  4995.0  801.31
  5005.0  801.31  5006.0  802.61  5009.8  803.90  5032.6  805.50  5048.0  807.52
  5061.1  809.82  5100.4  813.42  5129.1  816.54  5161.2  821.43  5175.7  823.18
  5197.4  827.06  5218.9  830.07  5232.4  832.70  5286.1  840.31  5295.6  841.38
#Mann=3,-1,0
  4648.8    0.09       0  4994.0    0.05       0  5006.0    0.09       0
#XS Ineff=2,0
       0                 5054.10    0.00  808.86
Permanent Ineff=
       F       F
Bank Sta=4994,5006
XS Rating Curve= 0
Exp/Cntr=0.5,0.3

Type RM Length L Ch R = 1,36929,122,122,122
BEGIN DESCRIPTION:
Kerr Creek 75.0
END DESCRIPTION:
XS GIS Cut Line= 4
      1499155.56       671805.06      1499483.31       671794.49
      1499593.25       671788.15      1499821.63       671650.70
#Sta/Elev= 30
  4667.5  836.60  4698.0  835.59  4721.8  833.92  4786.0  830.32  4845.1  825.71
  4893.2  821.35  4913.1  820.28  4930.0  817.54  4963.4  809.04  4979.9  807.92
  4998.0  799.55  4999.0  797.55  5001.0  797.55  5002.0  799.55  5026.4  804.20
  5036.9  804.78  5047.1  806.75  5055.8  808.98  5058.5  809.24  5090.7  809.13
  5128.2  809.94  5140.5  810.92  5164.9  812.06  5189.3  815.05  5230.9  818.79
  5259.4  822.15  5273.2  823.22  5291.4  825.88  5324.9  831.54  5372.1  837.72
#Mann=5,-1,0
  4667.5    0.09       0  4998.0    0.05       0  5002.0    0.09       0
  5047.1    0.13       0  5273.2    0.09       0
Bank Sta=4998,5002
XS Rating Curve= 0
Exp/Cntr=0.3,0.1

Type RM Length L Ch R = 1,36807,303,303,303
BEGIN DESCRIPTION:
Kerr Creek 74.5
END DESCRIPTION:
XS GIS Cut Line= 3
      1499347.23       671959.44      1499582.56       671891.39
      1499766.88       671724.08
#Sta/Elev= 30
  4837.8  827.27  4869.9  823.47  4878.3  822.73  4887.8  821.28  4906.3  819.50
  4933.6  816.32  4946.8  813.17  4958.7  809.84  4970.0  808.03  4981.0  807.33
  4985.0  804.95  4992.1  801.74  4995.8  799.42  4998.0  798.64  4999.0  796.64
  5001.0  796.64  5002.0  798.64  5008.1  799.72  5015.1  801.62  5028.2  807.44
  5083.1  807.41  5147.5  809.98  5163.5  809.56  5197.1  810.94  5211.7  811.09
  5227.2  812.15  5273.4  816.28  5304.2  818.08  5319.6  819.42  5331.7  821.31
#Mann=3,-1,0
  4837.8    0.13       0  4998.0    0.05       0  5002.0    0.13       0
Bank Sta=4998,5002
XS Rating Curve= 0
Exp/Cntr=0.3,0.1

Type RM Length L Ch R = 1,36504,493,493,493
BEGIN DESCRIPTION:
Kerr Creek 74.0
END DESCRIPTION:
XS GIS Cut Line= 3
      1499375.02       672125.01      1499552.11       672168.31
      1499928.23       672296.60
#Sta/Elev= 30
  4820.8  828.27  4838.7  826.43  4854.6  824.10  4875.6  821.73  4894.9  818.60
  4907.5  817.32  4947.1  808.83  4963.8  806.48  4978.3  803.70  4988.4  798.42
  4998.0  794.99  4999.0  792.99  5001.0  792.99  5002.0  794.99  5027.9  799.26
  5052.4  802.86  5065.0  803.03  5078.6  803.88  5090.7  804.04  5140.4  806.12
  5181.5  810.07  5203.0  812.98  5247.2  816.33  5256.2  817.51  5264.1  819.07
  5273.4  819.86  5287.8  823.62  5326.0  827.20  5380.4  834.23  5400.5  835.29
#Mann=3,-1,0
  4820.8    0.13       0  4998.0    0.05       0  5002.0    0.13       0
Bank Sta=4998,5002
XS Rating Curve= 0
Exp/Cntr=0.3,0.1

Type RM Length L Ch R = 1,36011,228,228,228
BEGIN DESCRIPTION:
Kerr Creek 73.0
END DESCRIPTION:
XS GIS Cut Line= 3
      1499224.98       672575.00      1499525.87       672612.07
      1499934.04       672635.40
#Sta/Elev= 30
  4699.6  845.46  4711.6  844.93  4736.5  842.57  4821.7  831.23  4838.3  828.71
  4894.9  818.63  4919.7  813.77  4967.8  801.16  4976.3  799.39  4983.5  796.38
  4989.8  795.04  4998.0  790.53  4999.0  788.53  5001.0  788.53  5002.0  790.53
  5005.5  791.23  5012.9  796.60  5038.0  798.84  5044.0  799.77  5065.5  800.29
  5103.6  800.93  5137.4  802.54  5166.6  805.25  5187.2  807.69  5233.6  815.56
  5257.0  817.04  5286.3  820.80  5303.2  822.26  5370.6  825.82  5411.6  828.65
#Mann=4,-1,0
  4699.6    0.13       0  4998.0    0.05       0  5002.0    0.13       0
  5065.5    0.09       0
Bank Sta=4998,5002
XS Rating Curve= 0
Exp/Cntr=0.3,0.1

Type RM Length L Ch R = 1,35783,448,448,448
BEGIN DESCRIPTION:
Kerr Creek 72.0
END DESCRIPTION:
XS GIS Cut Line= 3
      1499319.52       672813.36      1499561.18       672835.32
      1499940.09       672868.27
#Sta/Elev= 30
  4756.6  831.74  4786.6  831.57  4806.9  830.60  4837.3  826.89  4852.8  824.13
  4883.6  819.60  4895.9  817.05  4908.1  812.08  4924.5  802.91  4928.2  801.59
  4960.2  798.01  4981.5  798.03  4988.9  797.31  4996.9  792.83  4998.0  788.92
  4999.0  786.92  5001.0  786.92  5002.0  788.92  5004.8  791.18  5022.4  793.23
  5046.9  796.49  5099.4  798.46  5149.1  802.38  5165.6  804.25  5197.2  809.09
  5253.3  815.75  5282.2  818.08  5315.2  822.39  5331.7  823.06  5379.6  827.15
#Mann=4,-1,0
  4756.6    0.13       0  4998.0    0.05       0  5002.0    0.13       0
  5022.4    0.09       0
Bank Sta=4998,5002
XS Rating Curve= 0
Exp/Cntr=0.3,0.1

Type RM Length L Ch R = 1,35335,335,335,335
BEGIN DESCRIPTION:
Kerr Creek 71.0
END DESCRIPTION:
XS GIS Cut Line= 3
      1499103.12       673227.27      1499461.73       673265.17
      1499881.54       673305.99
#Sta/Elev= 30
  4638.6  818.78  4687.7  818.90  4712.4  816.81  4730.6  816.07  4769.4  809.59
  4785.5  808.32  4807.7  804.94  4849.1  801.39  4865.6  798.41  4894.6  795.32
  4925.9  793.63  4969.9  793.29  4988.9  787.52  4997.7  783.71  4998.0  782.03
  4999.0  780.03  5001.0  780.03  5002.0  782.03  5014.4  788.56  5040.1  793.38
  5139.3  794.86  5156.6  796.36  5176.8  796.68  5191.1  798.27  5238.5  809.19
  5264.9  813.26  5275.3  813.75  5334.5  819.79  5401.1  822.88  5421.0  822.77
#Mann=3,-1,0
  4638.6    0.09       0  4998.0   0.048       0  5002.0    0.09       0
Bank Sta=4998,5002
XS Rating Curve= 0
Exp/Cntr=0.3,0.1

Type RM Length L Ch R = 1,35000,482,482,482
BEGIN DESCRIPTION:
Kerr Creek 70.0
END DESCRIPTION:
XS GIS Cut Line= 3
      1499006.27       673607.83      1499422.66       673596.97
      1499845.67       673695.20
#Sta/Elev= 30
  4584.6  816.49  4600.6  815.18  4622.1  812.56  4676.9  806.92  4709.9  804.84
  4774.5  799.62  4789.2  799.21  4811.5  796.81  4832.4  795.21  4906.8  791.95
  4967.8  790.72  4990.1  789.23  4998.0  780.38  4999.0  778.38  5001.0  778.38
  5002.0  780.38  5020.5  787.73  5045.5  790.77  5084.8  789.92  5099.1  789.94
  5168.3  791.43  5185.7  793.89  5199.0  797.37  5203.7  798.02  5219.3  799.07
  5232.7  801.10  5282.2  806.15  5374.7  814.32  5389.8  814.57  5435.4  817.07
#Mann=4,-1,0
  4584.6    0.12       0  4622.1    0.09       0  4998.0   0.048       0
  5002.0    0.09       0
#XS Ineff=2,0
       0                 5073.00    0.00  790.70
Permanent Ineff=
       F       F
Bank Sta=4998,5002
XS Rating Curve= 0
Exp/Cntr=0.3,0.1

Type RM Length L Ch R = 1,34518,343,343,343
BEGIN DESCRIPTION:
Kerr Creek 69.0
END DESCRIPTION:
XS GIS Cut Line= 3
      1499001.95       673726.10      1499288.54       674016.82
      1499525.02       674225.02
#Sta/Elev= 30
  4595.5  812.23  4604.8  810.72  4618.7  810.04  4674.2  804.16  4709.9  801.40
  4720.0  799.52  4735.4  797.85  4765.8  791.29  4779.9  788.93  4803.0  787.32
  4821.7  787.28  4852.2  786.18  4882.6  786.66  4986.8  784.79  4992.4  781.76
  4997.5  779.89  4998.0  778.36  4999.0  776.36  5001.0  776.36  5002.0  778.36
  5003.7  780.66  5011.2  785.24  5064.5  789.85  5110.3  797.09  5171.6  804.45
  5177.7  804.50  5204.9  807.17  5245.5  812.37  5290.2  817.18  5318.8  818.89
#Mann=4,-1,0
  4595.5    0.12       0  4852.2    0.09       0  4998.0   0.048       0
  5002.0    0.09       0
Bank Sta=4998,5002
XS Rating Curve= 0
Exp/Cntr=0.3,0.1

Type RM Length L Ch R = 1,34175,319,319,319
BEGIN DESCRIPTION:
Kerr Creek 68.0
END DESCRIPTION:
XS GIS Cut Line= 3
      1498655.05       674169.76      1499099.89       674296.08
      1499429.35       674383.93
#Sta/Elev= 30
  4543.0  820.86  4560.0  820.93  4583.3  819.81  4609.0  817.68  4645.4  813.25
  4697.9  803.80  4739.1  795.28  4766.2  790.80  4815.5  784.09  4832.9  783.26
  4883.6  783.32  4958.5  783.06  4968.7  781.21  4993.3  779.37  4998.0  775.54
  4999.0  773.54  5001.0  773.54  5002.0  775.54  5011.3  780.41  5014.7  781.30
  5052.7  785.08  5062.2  785.36  5090.8  787.84  5136.5  792.99  5186.5  797.16
  5196.6  797.04  5242.4  801.21  5251.2  801.34  5327.2  807.71  5346.4  808.80
#Mann=4,-1,0
  4543.0    0.12       0  4883.6    0.09       0  4998.0   0.048       0
  5002.0    0.09       0
#XS Ineff=2,0
    0.00 4945.50  783.43               0
Permanent Ineff=
       F       F
Bank Sta=4998,5002
XS Rating Curve= 0
Exp/Cntr=0.3,0.1

Type RM Length L Ch R = 1,33856,376,376,376
BEGIN DESCRIPTION:
Kerr Creek 67.0
END DESCRIPTION:
XS GIS Cut Line= 3
      1498562.58       674661.17      1498994.06       674588.29
      1499380.09       674596.30
#Sta/Elev= 30
  4561.7  809.07  4611.1  806.89  4630.3  806.67  4654.0  805.65  4670.6  805.53
  4680.8  804.83  4706.9  804.01  4739.6  801.57  4754.1  801.19  4769.3  799.85
  4797.7  796.22  4825.9  790.67  4829.3  789.37  4844.3  785.81  4861.4  783.07
  4871.5  781.74  4894.7  781.30  4969.5  780.90  4994.9  776.22  4998.0  773.61
  4999.0  771.61  5001.0  771.61  5002.0  773.61  5018.8  778.14  5068.8  781.81
  5144.7  785.30  5188.6  791.23  5267.2  797.88  5332.1  801.77  5385.4  803.94
#Mann=4,-1,0
  4561.7    0.12       0  4894.7    0.09       0  4998.0   0.048       0
  5002.0    0.09       0
Bank Sta=4998,5002
XS Rating Curve= 0
Exp/Cntr=0.3,0.1

Type RM Length L Ch R = 1,33480,364,364,364
BEGIN DESCRIPTION:
Kerr Creek 66.0
END DESCRIPTION:
XS GIS Cut Line= 3
      1498578.19       675067.45      1499026.14       674928.83
      1499571.35       675051.29
#Sta/Elev= 30
  4531.9  826.62  4592.0  823.31  4640.5  818.32  4708.4  813.74  4713.4  812.14
  4738.0  807.60  4762.2  799.01  4772.0  794.70  4792.9  786.69  4816.2  781.44
  4826.9  780.45  4910.1  778.68  4980.3  778.92  4991.3  777.06  4993.7  774.16
  4998.0  771.73  4999.0  769.73  5001.0  769.73  5002.0  771.73  5010.0  773.32
  5026.4  774.94  5048.1  780.11  5078.7  782.21  5199.2  787.80  5268.7  796.88
  5323.6  802.29  5384.4  810.36  5491.8  827.14  5524.2  829.79  5559.6  831.05
#Mann=4,-1,0
  4531.9    0.12       0  4772.0    0.09       0  4998.0   0.048       0
  5002.0    0.09       0
Bank Sta=4998,5002
XS Rating Curve= 0
Exp/Cntr=0.3,0.1

Type RM Length L Ch R = 1,33116,613,613,613
BEGIN DESCRIPTION:
Kerr Creek 65.0
END DESCRIPTION:
XS GIS Cut Line= 3
      1498578.21       675332.03      1499166.09       675258.30
      1499611.03       675219.70
#Sta/Elev= 30
  4406.4  831.01  4418.1  829.68  4470.3  826.55  4564.9  816.08  4625.8  810.68
  4635.7  809.18  4710.0  803.80  4787.9  796.60  4814.2  794.37  4844.3  790.24
  4885.9  779.84  4898.4  777.74  4921.0  776.07  4947.2  777.65  4958.5  777.13
  4969.1  776.06  4998.0  770.77  4999.0  768.77  5001.0  768.77  5002.0  770.77
  5005.9  772.59  5032.1  777.62  5072.1  777.88  5083.8  778.81  5103.3  781.46
  5148.8  790.49  5244.7  803.33  5313.1  814.14  5376.8  822.86  5445.5  830.16
#Mann=4,-1,0
  4406.4    0.12       0  4787.9    0.09       0  4998.0   0.048       0
  5002.0    0.09       0
Bank Sta=4998,5002
XS Rating Curve= 0
Exp/Cntr=0.3,0.1

Type RM Length L Ch R = 1,32503,375,375,375
BEGIN DESCRIPTION:
Kerr Creek 64.0
END DESCRIPTION:
XS GIS Cut Line= 3
      1499298.99       676258.71      1499580.10       675695.64
      1499674.99       675475.02
#Sta/Elev= 30
  4367.1  798.95  4477.6  795.65  4538.8  792.28  4571.5  791.19  4599.2  789.82
  4663.9  787.72  4703.0  785.76  4757.3  781.55  4788.2  778.06  4837.4  773.89
  4860.7  773.35  4913.5  772.94  4963.7  774.00  4996.4  768.76  4997.0  768.13
  4998.0  766.13  5002.0  766.13  5003.0  768.13  5027.8  776.12  5035.8  781.28
  5045.5  788.82  5074.8  797.03  5084.3  802.22  5110.4  808.74  5120.0  811.70
  5132.5  814.01  5177.1  820.79  5190.3  823.11  5216.0  825.92  5236.6  826.96
#Mann=3,-1,0
  4367.1    0.09       0  4997.0   0.048       0  5003.0    0.09       0
Bank Sta=4997,5003
XS Rating Curve= 0
Exp/Cntr=0.5,0.3

Type RM Length L Ch R = 1,32128,103,103,103
BEGIN DESCRIPTION:
Corriher Springs Road (Kerr) us
END DESCRIPTION:
XS GIS Cut Line= 5
      1499479.32       676330.18      1499806.94       675968.24
      1499880.41       675914.31      1499941.11       675874.63
      1499956.71       675537.64
#Sta/Elev= 30
  4422.3  803.12  4523.7  798.86  4566.9  794.55  4681.8  784.95  4704.3  781.72
  4730.5  778.90  4823.7  773.04  4878.4  771.89  4976.9  773.34  4995.0  769.30
  4997.0  764.60  5003.0  764.60  5005.0  769.30  5042.6  771.74  5051.3  772.89
  5075.5  772.64  5105.5  774.74  5119.0  777.58  5130.3  781.60  5141.0  784.53
  5152.3  788.12  5165.6  793.39  5183.3  799.44  5214.6  807.63  5243.6  812.13
  5252.5  814.54  5288.3  818.53  5312.5  819.38  5392.3  826.59  5411.5  828.78
#Mann=3,-1,0
  4422.3    0.09       0  4995.0   0.048       0  5005.0    0.09       0
#XS Ineff=2,0
    0.00 4950.00  778.00 5050.00    0.00  778.00
Permanent Ineff=
       F       F
Bank Sta=4995,5005
XS Rating Curve= 0
Exp/Cntr=0.5,0.3

Type RM Length L Ch R =2,32084,,,
BEGIN DESCRIPTION:
Corriher Springs Road TOR (Kerr)
Structure ID: LDS_KC_07
Approximate Survey Structure
END DESCRIPTION:
Bridge Culvert--1,0,-1,-1,0
Deck Dist Width WeirC Skew NumUp NumDn MinLoCord MaxHiCord MaxSubmerge Is_Ogee
26.5,35,3,,24,24,,,,0,1,1,,,
  4416.1  4459.6  4511.9  4553.1  4590.7  4617.6  4644.7  4678.8  4729.9  4782.6
  4837.1  4890.6  5019.7  5062.1  5114.9  5158.8  5207.8  5275.0  5317.6  5376.0
  5428.5  5463.2  5495.5  5536.5
  802.97  800.35  797.15  793.44  790.67  788.78  786.09  783.00  780.07  777.90
  776.41  776.02  775.88  776.07  776.83  777.72  778.52  781.24  784.03  787.93
  791.93  795.09  798.90  804.23
  740.80  740.80  740.80  740.80  740.80  740.80  740.80  740.80  740.80  740.80
  740.80  740.80  740.80  740.80  740.80  740.80  740.80  740.80  740.80  740.80
  740.80  740.80  740.80  740.80
  4416.1  4459.6  4511.9  4553.1  4590.7  4617.6  4644.7  4678.8  4729.9  4782.6
  4837.1  4890.6  5019.7  5062.1  5114.9  5158.8  5207.8  5275.0  5317.6  5376.0
  5428.5  5463.2  5495.5  5536.5
  802.97  800.35  797.15  793.44  790.67  788.78  786.09  783.00  780.07  777.90
  776.41  776.02  775.88  776.07  776.83  777.72  778.52  781.24  784.03  787.93
  791.93  795.09  798.90  804.23
  740.62  740.62  740.62  740.62  740.62  740.62  740.62  740.62  740.62  740.62
  740.62  740.62  740.62  740.62  740.62  740.62  740.62  740.62  740.62  740.62
  740.62  740.62  740.62  740.62
Culvert=1,4.5,,35,0.012,0.2,1,1,3,764.6,5000,763.6,5000,Culvert #1,0,26.5
Culvert Bottom n=0.012
Culvert Bottom Depth=0
Culvert Depth Blocked=0
BC Design=,,0,,0,,,,,,

Type RM Length L Ch R = 1,32025,525,525,525
BEGIN DESCRIPTION:
Corriher Springs (Kerr) ds
END DESCRIPTION:
XS GIS Cut Line= 3
      1499579.18       676373.85      1499944.56       675993.04
      1500346.77       675765.41
#Sta/Elev= 30
  4466.8  802.03  4540.7  795.50  4596.5  789.29  4641.2  781.67  4679.6  777.90
  4731.8  775.13  4784.6  773.56  4891.6  772.26  4918.9  771.24  4974.3  771.29
  4990.0  769.92  4994.5  767.91  4995.0  768.30  4997.0  763.60  5003.0  763.60
  5005.0  768.30  5038.4  772.06  5123.4  774.57  5137.3  775.26  5151.9  777.20
  5192.0  778.59  5217.1  780.50  5242.2  783.42  5270.4  787.75  5292.8  789.79
  5321.6  793.97  5382.8  800.98  5403.1  801.88  5423.9  803.88  5456.7  808.04
#Mann=3,-1,0
  4466.8    0.09       0  4995.0   0.048       0  5005.0    0.09       0
#XS Ineff=2,0
    0.00 4956.30  775.95 5043.80    0.00  776.03
Permanent Ineff=
       F       F
Bank Sta=4995,5005
XS Rating Curve= 0
Exp/Cntr=0.5,0.3

Type RM Length L Ch R = 1,31500,487,487,487
BEGIN DESCRIPTION:
Kerr Creek 63.0
END DESCRIPTION:
XS GIS Cut Line= 3
      1499854.32       676597.92      1500341.08       676296.26
      1500720.10       676069.54
#Sta/Elev= 30
  4423.6  804.45  4541.1  796.67  4656.6  785.61  4670.7  785.34  4696.8  782.09
  4780.7  774.56  4873.4  769.18  4889.0  769.48  4920.1  768.03  4953.9  769.42
  4974.9  768.87  4989.8  766.23  4996.9  762.26  4997.0  760.55  4998.0  758.55
  5002.0  758.55  5003.0  760.55  5003.4  762.47  5007.2  767.88  5028.7  769.30
  5111.4  768.01  5136.8  769.63  5162.5  773.28  5198.3  782.14  5249.7  793.81
  5293.3  801.98  5336.7  811.42  5367.0  816.83  5399.6  821.40  5437.9  825.46
#Mann=4,-1,0
  4423.6    0.09       0  4997.0   0.048       0  5003.0    0.09       0
  5198.3    0.11       0
Bank Sta=4997,5003
XS Rating Curve= 0
Exp/Cntr=0.3,0.1

Type RM Length L Ch R = 1,31013,502,502,502
BEGIN DESCRIPTION:
Kerr Creek 62.0
END DESCRIPTION:
XS GIS Cut Line= 3
      1500405.25       676961.00      1500699.71       676619.90
      1500925.01       676374.98
#Sta/Elev= 30
  4553.7  797.79  4601.6  794.46  4655.0  791.74  4719.4  784.83  4757.8  779.03
  4822.7  770.43  4869.0  767.87  4938.5  766.23  4971.4  766.20  4989.3  765.01
  4997.0  758.13  4998.0  756.13  5002.0  756.13  5003.0  758.13  5004.3  759.80
  5026.6  766.69  5054.1  766.00  5077.3  766.83  5100.7  768.36  5121.5  774.51
  5139.4  781.72  5147.5  784.34  5153.0  785.25  5174.8  791.14  5200.1  796.08
  5219.4  799.28  5250.2  802.63  5264.9  805.24  5306.0  809.29  5337.1  811.40
#Mann=4,-1,0
  4553.7    0.09       0  4997.0   0.048       0  5003.0    0.09       0
  5077.3    0.11       0
Bank Sta=4997,5003
XS Rating Curve= 0
Exp/Cntr=0.3,0.1

Type RM Length L Ch R = 1,30511,507,507,507
BEGIN DESCRIPTION:
Kerr Creek 61.0
END DESCRIPTION:
XS GIS Cut Line= 3
      1500749.26       677287.59      1501061.24       676946.45
      1501463.62       676614.05
#Sta/Elev= 30
  4534.6  792.66  4624.4  785.72  4662.7  781.68  4701.6  779.03  4771.7  770.82
  4831.8  765.24  4899.6  764.45  4926.7  763.34  4968.1  763.82  4995.5  762.99
  4996.9  761.84  4997.0  757.25  4998.0  755.25  5002.0  755.25  5003.0  757.25
  5006.4  759.36  5010.6  760.20  5039.0  764.81  5051.0  765.62  5074.6  766.14
  5110.2  764.72  5152.4  766.01  5206.8  765.65  5247.5  768.57  5314.9  776.29
  5352.4  780.79  5378.8  782.84  5418.6  787.29  5442.4  790.91  5518.8  795.70
#Mann=4,-1,0
  4534.6    0.09       0  4997.0   0.048       0  5003.0    0.09       0
  5314.9    0.11       0
#XS Ineff=2,0
       0                 5098.00    0.00  766.13
Permanent Ineff=
       F       F
Bank Sta=4997,5003
XS Rating Curve= 0
Exp/Cntr=0.3,0.1

Type RM Length L Ch R = 1,30004,488,488,488
BEGIN DESCRIPTION:
Kerr Creek 60.0
END DESCRIPTION:
XS GIS Cut Line= 3
      1501249.03       677652.00      1501493.92       677188.44
      1501700.92       676893.99
#Sta/Elev= 30
  4474.5  784.30  4511.7  781.51  4576.3  775.12  4635.5  770.31  4772.2  763.31
  4814.5  762.05  4856.7  762.47  4893.4  760.74  4978.3  762.00  4982.4  759.54
  4995.5  757.24  4997.0  755.20  4998.0  753.20  5002.0  753.20  5003.0  755.20
  5009.0  756.24  5016.4  760.28  5037.3  761.83  5101.8  761.51  5146.9  762.44
  5179.7  763.62  5196.3  768.54  5217.0  777.57  5231.9  781.90  5261.2  789.07
  5275.5  791.39  5297.7  792.62  5303.4  793.54  5318.3  798.51  5358.7  801.10
#Mann=4,-1,0
  4474.5    0.09       0  4997.0   0.048       0  5003.0    0.09       0
  5146.9    0.11       0
Bank Sta=4997,5003
XS Rating Curve= 0
Exp/Cntr=0.3,0.1

Type RM Length L Ch R = 1,29516,503,503,503
BEGIN DESCRIPTION:
Kerr Creek 59.0
END DESCRIPTION:
XS GIS Cut Line= 3
      1501548.60       677850.04      1501864.21       677491.67
      1502147.68       677023.19
#Sta/Elev= 30
  4518.4  788.54  4536.8  787.22  4667.9  780.59  4745.8  774.70  4798.2  769.33
  4878.3  763.73  4921.4  759.96  4948.7  758.56  4976.8  759.44  4988.6  756.08
  4995.9  753.41  4997.0  752.05  4998.0  750.05  5002.0  750.05  5003.0  752.05
  5018.6  760.16  5117.2  759.13  5248.2  760.28  5261.2  760.38  5284.8  762.78
  5300.0  766.34  5316.5  774.43  5328.0  781.30  5350.1  791.85  5366.3  797.90
  5383.0  802.07  5416.7  809.42  5465.2  817.60  5522.5  824.81  5543.5  826.49
#Mann=4,-1,0
  4518.4    0.09       0  4997.0   0.048       0  5003.0    0.09       0
  5248.2    0.11       0
Bank Sta=4997,5003
XS Rating Curve= 0
Exp/Cntr=0.3,0.1

Type RM Length L Ch R = 1,29013,514,514,514
BEGIN DESCRIPTION:
Kerr Creek 58.0
END DESCRIPTION:
XS GIS Cut Line= 3
      1501524.96       678061.55      1501986.67       677966.92
      1502804.17       677649.70
#Sta/Elev= 30
  4526.4  794.49  4582.2  787.25  4612.8  783.89  4667.0  780.50  4739.9  773.97
  4782.0  766.18  4837.0  760.40  4898.3  757.69  4975.2  757.69  4993.3  754.61
  4994.1  749.21  4995.1  747.21  5004.9  747.21  5005.9  749.21  5016.2  753.76
  5035.3  758.09  5081.8  757.29  5143.2  757.65  5198.1  757.25  5218.3  758.21
  5376.7  759.20  5439.2  760.46  5606.7  767.17  5635.6  770.34  5688.0  772.30
  5724.9  774.54  5776.3  779.10  5813.5  780.04  5827.8  781.39  5874.6  783.37
#Mann=3,-1,0
  4526.4    0.09       0  4994.1   0.048       0  5005.9    0.09       0
Bank Sta=4994.1,5005.9
XS Rating Curve= 0
Exp/Cntr=0.3,0.1

Type RM Length L Ch R = 1,28499,485,485,485
BEGIN DESCRIPTION:
Kerr Creek 57.0
END DESCRIPTION:
XS GIS Cut Line= 5
      1501637.27       678866.54      1502011.66       678507.75
      1502123.70       678459.66      1502270.64       678390.32
      1502740.88       678520.19
#Sta/Elev= 30
  4359.2  773.07  4417.3  771.78  4478.7  771.52  4572.1  770.09  4657.1  768.17
  4697.6  766.12  4767.1  759.53  4808.6  757.22  4908.1  755.45  4965.1  755.56
  4983.0  754.40  4994.1  747.35  4995.1  745.35  5004.9  745.35  5005.9  747.35
  5010.6  756.18  5035.5  756.12  5109.3  754.16  5173.5  755.89  5249.2  759.04
  5275.0  759.08  5293.0  760.94  5347.5  768.75  5368.8  770.19  5391.7  774.04
  5424.5  775.66  5443.9  778.27  5477.9  779.72  5520.6  782.48  5650.0  787.01
#Mann=3,-1,0
  4359.2    0.09       0  4994.1   0.048       0  5005.9    0.09       0
Bank Sta=4994.1,5005.9
XS Rating Curve= 0
Exp/Cntr=0.3,0.1

Type RM Length L Ch R = 1,28014,513,513,513
BEGIN DESCRIPTION:
Kerr Creek 56.0
END DESCRIPTION:
XS GIS Cut Line= 3
      1501852.55       679022.37      1502266.57       678923.24
      1502630.98       678739.58
#Sta/Elev= 30
  4573.4  774.78  4672.3  771.66  4705.6  768.47  4750.5  763.14  4779.8  760.35
  4833.6  756.53  4872.6  754.86  4942.2  754.35  4986.5  753.44  4994.1  746.39
  4995.1  744.39  5004.9  744.39  5005.9  746.39  5015.4  747.39  5038.2  754.31
  5079.7  753.84  5099.8  753.02  5121.4  753.50  5188.1  753.66  5232.8  753.85
  5246.9  754.37  5259.9  756.19  5274.9  763.48  5300.4  774.00  5316.8  775.82
  5327.3  776.16  5342.2  778.12  5360.3  779.08  5379.6  779.37  5407.2  781.00
#Mann=5,-1,0
  4573.4    0.09       0  4994.1   0.048       0  5005.9    0.09       0
  5188.1    0.12       0  5360.3    0.09       0
Bank Sta=4994.1,5005.9
XS Rating Curve= 0
Exp/Cntr=0.3,0.1

Type RM Length L Ch R = 1,27501,498,498,498
BEGIN DESCRIPTION:
Kerr Creek 55.0
END DESCRIPTION:
XS GIS Cut Line= 3
      1501475.19       679466.63      1502359.87       679421.82
      1502990.66       679390.25
#Sta/Elev= 30
  4112.8  796.99  4250.4  791.14  4311.0  790.30  4396.7  780.81  4467.0  777.41
  4654.8  763.92  4690.1  763.33  4723.6  758.27  4753.9  755.70  4864.0  751.26
  4929.4  751.95  4965.8  752.48  4986.8  750.66  4994.1  744.85  4995.1  742.85
  5004.9  742.85  5005.9  744.85  5007.4  745.67  5026.1  745.94  5049.1  749.22
  5126.5  754.05  5144.7  757.71  5148.8  757.79  5196.4  769.71  5215.7  772.42
  5255.9  775.46  5429.7  781.26  5547.3  786.37  5589.1  790.01  5630.2  790.44
#Mann=5,-1,0
  4112.8    0.09       0  4929.4    0.12       0  4994.1   0.048       0
  5005.9    0.12       0  5429.7    0.09       0
Bank Sta=4994.1,5005.9
XS Rating Curve= 0
Exp/Cntr=0.3,0.1
